--- LFBUCKRV.prj (project) ---

Proj Title=LFBUCKRV
Current Plan=p01
Default Exp/Contr=0,0
English Units
Geom File=g01
Flow File=f01
Plan File=p01
BEGIN DESCRIPTION:
---------- MODELED AS PART OF WVEMD CTP PROGRAM, 2023----------
Stream Name: Left Fork Buckhannon River
Flood Zone:  AFH
Upshur County, WV
HEC-RAS Version: RAS 6.3
Vertical Datum: NAVD88
Projection: NAD 1983 StatePlane West Virginia S FIPS 4702 (US Feet)
Terrain: 1-meter LIDAR (FEMA Region III 3DEP collected 2016-2018)
Land Use: 2019 NLCD
Hydrologic Method:
WV 2010 Regional Regression Equations
Additional Model Notes:
Imported 3 shared XS's and snippet of streamline from Randolph model at upstream end
END DESCRIPTION:
DSS Export Rating Curves= 0
DSS Export Rating Curve Sorted= 0
DSS Export Volume Flow Curves= 0
DXF OffsetX= 0
DXF OffsetY= 0
DXF ScaleX= 0
DXF ScaleY= 0

--- LFBUCKRV.p01 (plan) ---

Plan Title=Floodplain
Program Version=6.31
Short Identifier=Floodplain
Geom File=g01
Flow File=f01
Subcritical Flow
K Sum by GR= 0
Std Step Tol= 0.01
Critical Tol= 0.01
Num of Std Step Trials= 20
Max Error Tol= 0.3
Flow Tol Ratio= 0.001
Split Flow NTrial= 30
Split Flow Tol= 0.02
Split Flow Ratio= 0.02
Log Output Level= 0
Friction Slope Method= 1
Unsteady Friction Slope Method= 2
Unsteady Bridges Friction Slope Method= 1
Parabolic Critical Depth
Global Vel Dist= 0 , 0 , 0
Global Log Level= 0
CheckData=True
Encroach Param=-1 ,0,0, 0
Mapping Interval=1HOUR
Computation Time Step Use Courant=        0
Computation Time Step Use Time Series=    0
Computation Time Step Count To Double=0
Computation Time Step Max Doubling=0
Computation Time Step Max Halving=0
Computation Time Step Residence Courant=0
Run HTab= 0
Run UNet= 0
Run Sediment= 0
Run PostProcess= 0
Run WQNet= 0
Run RASMapper=-1
UNET Theta= 0
UNET Theta Warmup= 0
UNET ZTol= 0
UNET ZSATol= 0
UNET MxIter= 0
UNET Max Iter WO Improvement= 0
UNET MaxInSteps= 0
UNET DtIC= 0
UNET DtMin= 0
UNET MaxCRTS= 0
UNET WFStab= 0
UNET SFStab= 0
UNET WFX= 1
UNET SFX= 1
UNET Gravity=32.17405
UNET 1D Methodology=Finite Difference
UNET DSS MLevel= 1
UNET Pardiso=0
UNET DZMax Abort= 0
UNET Use Existing IB Tables= 0
UNET Froude Reduction=False
UNET Froude Limit= 0
UNET Froude Power= 0
UNET D1 Cores= 0
UNET WindReference=Eulerian
UNET WindDragFormulation=Hsu (1988)
UNET D2 Coriolis=0
UNET D2 Cores= 0
UNET D2 Theta= 1
UNET D2 Theta Warmup= 1
UNET D2 Z Tol= 0.01
UNET D2 Volume Tol= 0.01
UNET D2 Max Iterations= 20
UNET D2 Equation= 0
UNET D2 RampUpFraction=0.1
UNET D2 TimeSlices= 1
UNET D2 Turbulence Formulation=Non-Conservative (original)
UNET D2 Eddy Viscosity=0.3
UNET D2 Transverse Eddy Viscosity=0.1
UNET D2 Smagorinsky Mixing=0
UNET D2 BCVolumeCheck=0
UNET D2 Cores=0
UNET D2 SolverType=PARDISO (Direct)
UNET D2 Minimum Iterations= 3
UNET D2 Maximum Iterations= 30
UNET D2 Restart Number= 10
UNET D2 Relaxation Coeff=1.3
UNET D2 SOR Precondition Iterations= 10
UNET D2 ILUT Maximum Fill= 8
UNET D2 ILUT Tolerance=1E-08
UNET D2 Convergence Tolerance=0.00001
UNET D1D2 MaxIter= 0
UNET D1D2 ZTol=0.01
UNET D1D2 QTol=0.1
UNET D1D2 MinQTol=1
Write IC File= 0
Write IC File at Fixed DateTime=0
Write IC File at Sim End=0
Echo Input=False
Echo Parameters=False
Echo Output=False
Write Detailed= 0
HDF Write Warmup=0
HDF Write Time Slices=0
HDF Flush=0
HDF Compression= 1
HDF Chunk Size= 1
HDF Spatial Parts= 1
HDF Use Max Rows=0
HDF Fixed Rows= 1
Calibration Method= 0
Calibration Iterations= 20
Calibration Max Change=0.05
Calibration Tolerance=0.2
Calibration Maximum=1.5
Calibration Minimum=0.5
Calibration Optimization Method= 1
WQ AD Non Conservative
WQ ULTIMATE=-1
WQ Max Comp Step=1HOUR
WQ Output Interval=15MIN
WQ Output Selected Increments= 0
WQ Create Restart=0
WQ Fixed Restart=0
WQ System Summary=0
WQ Write To DSS=0
Sorting and Armoring Iterations= 10
XS Update Threshold= 0.02
Bed Roughness Predictor= 0
Hydraulics Update Threshold= 0.02
Energy Slope Method= 1
Volume Change Method= 1
Sediment Retention Method= 0
Sediment TS Multiplier= 1
Warm Up Method= 0
XS Weighting Method= 0
Number of US Weighted Cross Sections= 1
Number of DS Weighted Cross Sections= 1
Upstream XS Weight=0
Main XS Weight=1
Downstream XS Weight=0
Number of DS XS's Weighted with US Boundary= 1
Upstream Boundary Weight= 1
Weight of XSs Associated with US Boundary= 0
Number of US XS's Weighted with DS Boundary= 1
Downstream Boundary Weight= 0.5
Weight of XSs Associated with DS Boundary= 0.5
Percentile Method= 0
Sediment Output Level= 3
Mass or Volume Output= 0
Output Increment Type= 1
Profile and TS Output Increment= 1
Transport Output Increment 1
XS Output Flag= 0
XS Output Increment= 10
Read HDF5 Sediment Hotstart= 0
Sediment Hotstart Type= 0
Write Gradation File= 0
Read Gradation Hotstart= 0
Write HDF5 File= 1
Write Binary Output= 1
Write DSS Sediment File= 0
DSS Sediment Output Type= 1
SV Curve= 0
Specific Gage Flag= 0
Subcell Erosion Methods= 0
Subcell Deposition Methods= 0
Advection Scheme= 1
Matrix Solver= 0
Implicit Weighting Factor= 1
Maximum Outer Loop Convergence Iterations= 5
Convergence Maximum Absolute= 0.001
Convergence RMSE= 0.0001
Grain Fractions Max Abs Error= 0.001
Max Subgrid Regions= 1
Max Subgrid Length Scale= 3.402823E+38
Initial Layer Thickness= 3.402823E+38
Min Layer Thickness= 3.402823E+38
Max Layer Thickness= 3.402823E+38
Number of Layers= 5

--- LFBUCKRV.f01 (steady flow) ---

Flow Title=Flows
Program Version=6.31
Number of Profiles= 1
Profile Names=01pct
River Rch & RM=LFBUCKRV,Main,34765
    4710
River Rch & RM=LFBUCKRV,Main,20421
    5350
Boundary for River Rch & Prof#=LFBUCKRV,Main            , 1
Up Type= 0
Dn Type= 3
Dn Slope=0.00442
DSS Import GetInterval= 0
DSS Import GetPeak= 0
DSS Import FillOption= 0

--- LFBUCKRV.g01 (geometry) ---

Geom Title=Geometry
Program Version=6.31

River Reach=LFBUCKRV        ,Main
Reach XY= 30
2213036.24817476636616.130237758     2212455.677637854.243000001
2211099.37500001 638187.738000022209831.66900001639313.736000001
2209770.37199999639650.1210000072208509.47700001640207.797999993
2208439.36700001640787.3940000092209269.09900004641562.555000007
2209175.03700002641950.7360000012208363.56199999 641962.21100001
2207540.81200004641552.5680000042205955.83700003642982.613999993
     2205314.572644699.2539999932204542.32999998      645588.022
2202539.49800003645518.9130000032201914.05800001646428.171000004
      2199182.08646313.9050000012197871.39200002647443.594000012
     2197910.654648085.8889999992197421.94300003648630.716999993
     2196536.609647827.3970000152196253.87900001647080.394999996
2195741.21699999646851.0639999962195039.71500002647035.553000018
2194209.52500005647510.4710000162193414.47499998 648649.26000002
2192770.09200002648448.7740000192192128.05400003648864.999000013
2191294.23000003650260.7919999962190223.54794142650454.868443087

Type RM Length L Ch R = 1 ,34765   ,289.3,297.4,311.4
XS GIS Cut Line= 2
2212781.51854692636706.0752715142213268.32829419636725.659571691
#Sta/Elev= 30
       0 2205.45    14.7 2196.56    42.7  2187.1    54.7 2184.54    70.7 2182.96
   122.8 2174.82   150.8 2165.21   162.8 2165.32   174.8 2162.91   198.8 2161.88
   210.8 2157.66   221.1 2155.17   236.4 2153.44   278.9 2153.44   282.9 2153.83
  285.752155.204   294.9 2161.52   306.9 2172.91   318.9 2181.08   334.9 2193.71
   346.9 2200.34   355.7 2203.07   374.9 2211.61     387 2214.58     399 2219.65
   413.5  2223.6   444.3 2234.13   459.7 2240.78     471 2248.02   487.2 2248.87
#Mann= 3 ,-1,0
       0      .1       0   221.1    .045       0  285.75      .1       0
Bank Sta=221.1,285.75
XS Rating Curve= 0 ,0
Exp/Cntr(USF)=0,0
Exp/Cntr=0.3,0.1

Type RM Length L Ch R = 1 ,34467   ,252.5,253.6,255.2
XS GIS Cut Line= 2
 2212721.2749462636910.6239836612213177.30936461637095.275956762
#Sta/Elev= 30
       0 2199.51     3.1 2198.22    16.1 2197.54    31.8 2188.55      42 2183.78
    47.2 2182.54   102.4    2172   132.6 2165.01   145.5 2164.86   162.8  2160.6
   171.4 2161.86   180.1 2161.72   191.6 2157.69   201.6 2152.15  208.592149.914
   214.6 2148.42   253.4 2148.15   262.1 2148.26   271.4  2149.9   283.7 2151.16
   296.6 2155.24   309.5 2156.46   317.5 2158.55   331.1 2168.28   339.7 2175.81
   357.4  2186.3   431.2 2203.38   447.6 2208.72   456.3 2210.46     492 2220.95
#Mann= 3 ,-1,0
       0      .1       0  208.59    .045       0   271.4      .1       0
Bank Sta=208.59,271.4
XS Rating Curve= 0 ,0
Exp/Cntr(USF)=0,0
Exp/Cntr=0.3,0.1

Type RM Length L Ch R = 1 ,34214   ,314.4,318.2,324.2
XS GIS Cut Line= 2
2212665.31980283   637153.7712662213040.21926337637321.636696092
#Sta/Elev= 30
       0 2179.71     7.5 2175.87      25 2168.61      35 2165.27    51.3 2161.75
    59.2 2159.22   107.7 2158.48   116.7 2159.66   121.5 2158.61   137.9 2159.37
   152.1 2158.43   156.5 2157.63   160.9 2154.79   165.3 2150.74  170.31 2147.61
   177.3 2146.32   222.3 2146.09   234.8 2146.33   239.82147.656   262.1 2154.99
   274.9 2160.61   292.4 2171.75   296.8 2175.48   305.5 2184.62   311.8 2187.98
   318.7 2189.31   337.7 2190.15   366.9 2193.83   393.2  2195.9   410.8 2198.36
#Mann= 3 ,-1,0
       0      .1       0  170.31    .045       0   239.8      .1       0
Bank Sta=170.31,239.8
XS Rating Curve= 0 ,0
Exp/Cntr(USF)=0,0
Exp/Cntr=0.3,0.1

Type RM Length L Ch R = 1 ,33895   ,253.8,256.4,259.8
XS GIS Cut Line= 2
2212496.75087049637388.8779414462212827.72636404637597.772310326
#Sta/Elev= 30
       0 2183.51     8.8 2183.53    20.1 2178.51    32.4 2175.26    40.4 2171.55
    84.5 2157.16    90.5  2156.4   107.1 2156.32   131.8 2154.98   147.7 2156.14
   156.4 2154.73   176.7 2153.89   188.5 2150.56   202.8 2149.17   210.4  2145.2
   214.22144.166   221.6 2143.31   259.5 2143.24   278.2 2143.31  282.832144.214
   286.9  2147.2   292.8 2152.96   301.4 2159.32     313 2168.93   321.7 2174.94
   325.7 2177.04   339.1 2180.08   349.3 2180.07     373 2181.89   391.4 2184.95
#Mann= 3 ,-1,0
       0      .1       0   214.2    .045       0  282.83      .1       0
Bank Sta=214.2,282.83
XS Rating Curve= 0 ,0
Exp/Cntr(USF)=0,0
Exp/Cntr=0.3,0.1

Type RM Length L Ch R = 1 ,33639   ,275.8,284.5,293.3
XS GIS Cut Line= 2
2212354.99026604637575.0303100992212654.77117812637804.517766929
#Sta/Elev= 30
       0 2178.44     5.2 2178.29     8.1 2177.24    16.6 2170.63    21.6 2167.76
    36.8 2160.98    45.2  2158.7      67 2156.89    92.2 2151.62   133.6 2152.09
   141.7 2153.58   147.6 2153.78   157.7 2152.64   167.9 2152.56   182.1  2150.2
   192.9 2149.46     208 2144.97   222.1 2143.36   228.2 2141.14   253.4 2140.75
  293.192141.142   298.7 2144.65   308.8 2155.27   313.8 2157.83   319.4 2158.72
   323.9  2157.3   332.6  2152.5   336.2 2152.47   365.5 2156.99   377.5 2160.12
#Mann= 3 ,-1,0
       0      .1       0   228.2    .045       0  293.19      .1       0
Bank Sta=228.2,293.19
XS Rating Curve= 0 ,0
Exp/Cntr(USF)=0,0
Exp/Cntr=0.3,0.1

Type RM Length L Ch R = 1 ,33354   ,304.6,311,317.2
XS GIS Cut Line= 2
2212213.94732641637737.9067303912212444.54500634638043.863129255
#Sta/Elev= 30
       0 2169.54    24.1 2161.67    54.2 2155.69    63.9 2155.51    69.2  2154.5
      81 2149.92    89.2 2147.93   109.3 2147.36   114.3 2148.19   119.3  2150.5
   134.3 2148.89   139.3  2149.4   146.7 2151.43   155.3 2151.76   166.7 2149.51
   174.4 2146.37  200.742139.271   204.5 2138.55   224.5 2138.34   254.5 2138.52
   264.6  2139.3   269.6 2140.19   275.3 2142.18   278.1 2144.73   289.5 2157.96
   294.6  2160.7   324.7 2164.06   359.7 2164.72   379.8 2163.87   383.1 2164.87
#Mann= 3 ,-1,0
       0      .1       0  200.74    .045       0   264.6      .1       0
Bank Sta=200.74,264.6
XS Rating Curve= 0 ,0
Exp/Cntr(USF)=0,0
Exp/Cntr=0.3,0.1

Type RM Length L Ch R = 1 ,33044   ,213.8,218.7,224.6
XS GIS Cut Line= 2
2212002.41752579637911.8417173852212154.65055716638219.126910339
#Sta/Elev= 30
       0 2154.39     5.3 2153.95    14.2 2151.63    20.2 2150.57    37.2 2149.58
    41.7 2149.82    50.6 2147.53    55.1 2148.47      65 2148.65    72.9 2147.95
    94.1  2148.1   121.7 2146.52   135.4 2142.81   148.1 2138.14  156.562136.198
   162.2  2135.5   171.1 2135.28   211.2 2135.19   229.2 2136.19   229.2  2136.2
   235.1 2137.57   242.5 2140.27   251.5 2141.98   255.9 2143.28   276.9 2156.15
   288.9 2162.83   296.1 2166.11   309.5  2170.9   328.3 2175.94   342.9 2177.84
#Mann= 3 ,-1,0
       0      .1       0  156.56    .045       0   229.2      .1       0
Bank Sta=156.56,229.2
XS Rating Curve= 0 ,0
Exp/Cntr(USF)=0,0
Exp/Cntr=0.3,0.1

Type RM Length L Ch R = 1 ,32825   ,153.1,157.4,160.7
XS GIS Cut Line= 2
 2211845.9557991637995.0060585972211919.25318458638302.291251552
#Sta/Elev= 30
       0 2145.89    10.5 2143.84    22.8 2144.67    35.1 2143.68    47.5  2145.8
    63.9 2147.04    80.4 2149.17    93.3 2149.98    96.8 2149.56   109.2 2142.58
   113.2 2141.32   126.5 2141.57   136.5 2140.41   150.3 2137.13   161.9 2132.75
   199.6 2132.04  202.032132.769   203.7 2133.27   207.8 2135.47     212 2136.68
   224.3 2137.45   232.5 2135.67   236.1 2135.54   240.7 2135.73     246 2136.77
   265.4  2145.9   277.8 2153.73   298.3 2169.18   306.5 2175.83   315.9 2182.23
#Mann= 3 ,-1,0
       0      .1       0   161.9    .045       0  202.03      .1       0
Bank Sta=161.9,202.03
XS Rating Curve= 0 ,0
Exp/Cntr(USF)=0,0
Exp/Cntr=0.3,0.1

Type RM Length L Ch R = 1 ,32667   ,102.9,130.6,156.8
XS GIS Cut Line= 3
2211822.38765986638085.0667734482211730.33808019638139.518637481
2211740.70986381638332.693107501
#Sta/Elev= 30
       0 2146.54    31.6 2146.42    58.3 2145.42    71.8 2141.69    86.2 2139.91
    94.5 2140.74   102.4 2143.21   112.6 2143.58   116.6  2142.5   120.6 2140.56
   132.6 2132.72   136.7 2131.49   163.5 2130.35   176.7 2130.58   180.7 2131.83
  181.612132.708   184.7 2135.69   188.7 2142.53   192.7 2147.84   205.3 2159.98
   212.8 2166.03   221.1 2173.65   228.1  2180.7   231.9 2183.32   236.8 2185.72
   244.8 2188.48   264.8 2194.19   272.8 2194.86   285.1  2199.3   300.4 2203.66
#Mann= 3 ,-1,0
       0      .1       0   132.6    .045       0  181.61      .1       0
Bank Sta=132.6,181.61
XS Rating Curve= 0 ,0
Exp/Cntr(USF)=0,0
Exp/Cntr=0.3,0.1

Type RM Length L Ch R = 1 ,32537   ,49.1,56.9,58.4
XS GIS Cut Line= 3
2211809.18729333638058.8198900442211512.33288215 638217.39596439
2211579.56913768638339.182389488
#Sta/Elev= 30
       0 2142.48      39 2141.61   105.5 2137.83   132.6 2139.11   141.7 2141.15
   146.3 2141.65   155.3 2141.42   159.9 2142.39   165.1  2141.5   173.9 2137.09
   188.7 2134.16  203.662129.782   234.2 2129.29  257.452129.762   268.7 2132.66
   280.3    2133   286.8 2134.09   295.1 2134.42   318.6 2138.81   327.6 2139.51
   336.6 2139.14   340.9 2141.17   344.5 2141.89   363.7 2142.19   377.5 2143.84
   391.1 2148.67   430.5 2169.58   441.4 2170.89   450.5 2175.69   475.7 2182.82
#Mann= 3 ,-1,0
       0      .1       0  203.66    .045       0  257.45      .1       0
Bank Sta=203.66,257.45
XS Rating Curve= 0 ,0
Exp/Cntr(USF)=0,0
Exp/Cntr=0.3,0.1

Type RM Length L Ch R = 1 ,32480   ,155.3,119.4,89.7
XS GIS Cut Line= 3
2211755.90573235638035.3506310412211459.05132117638193.926705387
 2211526.2875767638315.713130485
#Sta/Elev= 30
       0 2144.83    37.8 2143.23    46.3 2142.24    58.6 2138.71    66.2 2138.01
    97.3 2139.39   119.4 2136.28   135.7 2136.74   148.2 2133.98   158.4  2133.3
     172 2127.87  184.772126.665     214 2125.73   257.8 2126.68   285.4 2131.75
   321.7 2136.27   335.6 2139.47   342.7 2137.97   354.5  2137.7   363.3 2134.74
   376.8 2134.86   381.4  2135.7   390.5 2141.18   398.7 2143.99   404.2 2144.46
   413.4 2142.03   427.1 2143.58   439.9 2146.73   449.9 2150.46   475.7 2166.37
#Mann= 3 ,-1,0
       0      .1       0  184.77    .045       0   257.8      .1       0
#XS Ineff= 2 , 0
                          337.46         2147.95
Permanent Ineff=
       F       F
Bank Sta=184.77,257.8
XS Rating Curve= 0 ,0
Exp/Cntr(USF)=0,0
Exp/Cntr=0.3,0.1

Type RM Length L Ch R = 1 ,32361   ,166.4,164.2,162.5
XS GIS Cut Line= 3
2211439.92813868637986.5348290082211441.22461163638216.010541717
2211512.53062405638315.838959111
#Sta/Elev= 30
       0 2165.13     2.9 2164.08    18.5 2155.83    26.6 2152.74    50.6 2141.66
    62.6 2136.89    86.6 2131.91   106.6 2126.74   114.6 2127.46  119.982126.137
   122.6 2125.34   138.6 2124.65   150.6 2125.22   155.92126.082   162.6 2127.91
   174.6 2129.27   198.6 2138.16   209.7 2140.14   234.6 2140.51   238.2  2139.2
   245.7 2135.05   260.4 2134.88   265.3 2135.91   275.4 2141.04   281.2  2142.4
     285 2142.67   294.8 2141.51   315.6 2142.96   319.4 2143.86   352.2  2162.5
#Mann= 3 ,-1,0
       0      .1       0  119.98    .045       0   155.9      .1       0
Bank Sta=119.98,155.9
XS Rating Curve= 0 ,0
Exp/Cntr(USF)=0,0
Exp/Cntr=0.3,0.1

Type RM Length L Ch R = 1 ,32196   ,361.6,340,317.6
XS GIS Cut Line= 3
2211267.49142336637997.9266774952211289.05776948638290.975262887
2211393.08367425638410.224470795
#Sta/Elev= 30
       0 2172.29    35.3 2166.46    51.4    2162    79.5 2138.93    91.5 2127.55
   100.8 2125.18   139.6 2124.61   160.6 2125.16   167.7 2126.06   179.7 2130.68
   187.8 2132.53   207.8 2133.73   231.9 2132.63   239.9 2133.02   251.9  2135.7
     276  2137.4     284 2141.04     288 2141.71   304.7 2139.94   316.8 2134.82
   323.3 2133.31   337.3 2134.74   347.3 2134.83   357.1 2137.54   365.8 2136.69
   374.2 2137.62   391.2 2140.69   399.7 2143.96   426.4 2157.08   452.1 2172.25
#Mann= 3 ,-1,0
       0      .1       0   100.8    .045       0   160.6      .1       0
Bank Sta=100.8,160.6
XS Rating Curve= 0 ,0
Exp/Cntr(USF)=0,0
Exp/Cntr=0.3,0.1

Type RM Length L Ch R = 1 ,31856   ,297.9,299.1,299.7
XS GIS Cut Line= 2
2210908.47519105638222.4703987692211211.67264519638479.997943507
#Sta/Elev= 30
       0 2173.29    10.1 2164.33    27.2 2151.26    52.1 2134.77    64.1 2124.07
      67 2122.56    69.8 2121.76   80.832120.255   106.7 2119.49   127.8 2119.82
  131.622120.302   141.3 2122.68   151.8 2126.98   154.9 2127.73   164.8 2128.91
     189 2130.67     241 2131.48   246.3 2131.21   254.3 2132.85   256.8 2132.87
   263.7 2131.78   313.9 2130.69   322.4 2129.96   330.2 2130.29   339.4 2131.61
   350.8 2131.16   361.7  2134.3   368.7 2135.62   387.3 2145.14   397.8  2151.6
#Mann= 3 ,-1,0
       0      .1       0   80.83    .045       0  131.62      .1       0
Bank Sta=80.83,131.62
XS Rating Curve= 0 ,0
Exp/Cntr(USF)=0,0
Exp/Cntr=0.3,0.1

Type RM Length L Ch R = 1 ,31557   ,272.4,278.3,283.1
XS GIS Cut Line= 2
2210714.37807605638445.7455114492211046.75352787638695.661404618
#Sta/Elev= 30
       0  2158.4     9.4 2151.57    17.3 2146.73    40.9 2129.75    43.7 2127.08
    49.4 2120.17    52.3 2118.03   56.522117.472    66.6 2116.87    85.6 2117.47
    95.1 2118.11   135.1 2117.77   146.6  2120.2   167.4 2121.18   198.7 2125.86
     212 2126.57   232.5 2126.13   252.3 2127.06   287.5 2123.35   292.3 2123.62
   307.5 2126.25   323.7 2125.17   335.1 2126.01   343.7 2127.87   352.6 2130.89
   360.8 2135.45   380.8 2148.42   387.6 2152.04   398.4 2156.29   415.9 2160.53
#Mann= 3 ,-1,0
       0      .1       0   56.52    .045       0    85.6      .1       0
#XS Ineff= 2 , 0
                          252.35          2128.6
Permanent Ineff=
       F       F
Bank Sta=56.52,85.6
XS Rating Curve= 0 ,0
Exp/Cntr(USF)=0,0
Exp/Cntr=0.3,0.1

Type RM Length L Ch R = 1 ,31279   ,309.2,312.7,313.5
XS GIS Cut Line= 2
2210521.94150222638617.9177983472210810.04191468638954.357206196
#Sta/Elev= 30
       0 2156.31     9.6 2148.93    34.2  2125.6    41.2 2120.32    46.5    2118
    52.6 2117.09    60.6 2114.69    71.1 2114.05    95.7  2113.5  126.752114.055
   138.7 2115.62   157.2 2114.29   172.8 2116.73   183.3 2120.86   188.3 2121.81
     236 2121.75   247.9 2123.78   259.2 2120.82   278.1 2117.34   293.3 2120.55
   329.4 2118.26   355.7 2120.14   369.9 2122.26   378.4  2125.4     397 2136.85
   409.6 2148.08   415.2 2153.89   420.9 2158.29   430.9 2167.63   442.9 2175.77
#Mann= 3 ,-1,0
       0      .1       0    71.1    .045       0  126.75      .1       0
#XS Ineff= 2 , 0
                          248.62         2130.48
Permanent Ineff=
       F       F
Bank Sta=71.1,126.75
XS Rating Curve= 0 ,0
Exp/Cntr(USF)=0,0
Exp/Cntr=0.3,0.1

Type RM Length L Ch R = 1 ,30966   ,305.6,304,303.1
XS GIS Cut Line= 2
2210292.71798612638813.1686684882210533.91023747639129.537725455
#Sta/Elev= 30
       0 2147.07     5.3 2145.95    10.1 2143.63    32.1 2131.25    51.9 2121.13
    62.4 2113.11    65.4 2111.19    68.1 2110.43    80.5 2109.53   104.7 2109.46
   139.5 2109.78   148.12110.438     166 2112.62   176.6 2114.88   216.3 2116.36
   226.4 2117.66   230.8 2117.22   253.6 2112.82   271.6 2114.71   276.5 2114.44
   286.7 2112.76   289.4 2112.85   309.2 2121.32   322.4 2123.91   350.7 2141.74
   357.1 2146.42     362 2149.18   373.5 2154.19   381.8 2156.51   397.8 2162.37
#Mann= 3 ,-1,0
       0      .1       0    68.1    .045       0   148.1      .1       0
#XS Ineff= 2 , 0
                          226.18         2124.95
Permanent Ineff=
       F       F
Bank Sta=68.1,148.1
XS Rating Curve= 0 ,0
Exp/Cntr(USF)=0,0
Exp/Cntr=0.3,0.1

Type RM Length L Ch R = 1 ,30662   ,320.2,316.5,314.5
XS GIS Cut Line= 2
2210048.39336787638999.5444990782210281.75470197639287.722253939
#Sta/Elev= 30
       0 2152.92    12.4  2144.9    27.8 2133.57    38.1 2127.64    49.4 2120.08
    52.2 2117.28    57.9 2109.86   61.272107.297    63.6 2106.49    80.6 2107.15
   114.8 2105.88   135.9 2105.97  143.532107.258   152.2 2110.23   158.6 2111.36
   196.7 2111.58   215.8 2110.33   228.5 2111.57   234.8 2110.23   251.3 2109.33
   271.2 2110.51   285.4 2108.55   302.5 2110.66   316.1 2110.41   323.8  2114.4
   336.7 2123.57   349.2 2133.84   355.6 2136.49     365 2141.76   370.8 2143.65
#Mann= 3 ,-1,0
       0      .1       0   61.27    .045       0  143.53      .1       0
Bank Sta=61.27,143.53
XS Rating Curve= 0 ,0
Exp/Cntr(USF)=0,0
Exp/Cntr=0.3,0.1

Type RM Length L Ch R = 1 ,30346   ,416.8,407.7,404.9
XS GIS Cut Line= 2
2209800.93638272639212.5454483232210107.90833898639516.385037687
#Sta/Elev= 30
       0 2127.92     8.4 2120.94    19.7 2113.33    23.6 2111.28    32.7  2109.3
    46.4 2109.37    49.6 2108.07    56.5 2103.04    60.8 2102.45    83.3 2102.03
   114.6 2103.01     126 2105.86     134 2106.87   177.2 2107.55   200.7 2108.64
   217.7 2108.29   226.2  2106.6   237.5 2107.52   251.6 2105.05   290.9 2107.33
   330.7 2106.68   347.9 2108.37   367.6 2104.94   381.8 2104.98   384.6 2106.53
   387.3 2108.83   393.2 2116.12   398.7 2120.87     410 2129.46   431.9 2144.38
#Mann= 3 ,-1,0
       0      .1       0    56.5    .045       0   114.6      .1       0
Bank Sta=56.5,114.6
XS Rating Curve= 0 ,0
Exp/Cntr(USF)=0,0
Exp/Cntr=0.3,0.1

Type RM Length L Ch R = 1 ,29938   ,153.6,161.8,172
XS GIS Cut Line= 3
2209626.87553733639389.3833879732209701.43569687639575.258715268
2209870.50873469639777.936332035
#Sta/Elev= 30
       0 2109.81     8.4 2106.07    21.3 2104.45    42.9 2104.65    59.3 2106.58
    68.5 2106.76   116.1 2105.76   133.4 2103.19   173.1 2104.81   214.9  2105.4
   223.6 2104.88   237.7 2102.46   254.9  2102.1   285.7 2097.83   291.6 2097.12
   308.7 2096.86     320 2097.76   322.9 2098.81   328.5 2103.76     333 2106.44
   343.4  2107.3   348.2 2109.69     359 2122.71   373.1 2136.64   390.3 2148.21
   393.9 2149.74   400.7 2151.11   411.1 2158.01   421.6 2162.73   464.2 2184.46
#Mann= 3 ,-1,0
       0      .1       0   285.7    .045       0     320      .1       0
#XS Ineff= 2 , 0
          214.08 2128.47
Permanent Ineff=
       F       F
Bank Sta=285.7,320
XS Rating Curve= 0 ,0
Exp/Cntr(USF)=0,0
Exp/Cntr=0.3,0.1

Type RM Length L Ch R = 1 ,29776   ,283.6,278.3,275.7
XS GIS Cut Line= 2
2209572.27359897639394.2227285612209625.52383628639823.356993952
#Sta/Elev= 30
       0 2123.78    23.1 2116.78    39.3 2109.63    51.3 2105.83    63.4 2103.66
    91.7 2103.56    95.7 2103.81   103.7 2105.88   107.8 2105.85   124.5 2104.98
   138.8 2101.81   144.1 2101.39   156.7 2102.25   172.3 2101.75   192.4 2103.21
   216.6 2103.79   232.7 2102.01   244.8 2097.65     250  2096.8     265 2097.07
   285.8 2095.75   301.2 2095.07   313.3  2095.8   333.5 2103.28     354 2105.13
   365.7 2111.53   390.1 2120.75   410.1 2130.37   418.1 2133.07   432.4 2139.33
#Mann= 3 ,-1,0
       0      .1       0   285.8    .045       0   313.3      .1       0
#XS Ineff= 2 , 0
          186.47 2108.35
Permanent Ineff=
       F       F
Bank Sta=285.8,313.3
XS Rating Curve= 0 ,0
Exp/Cntr(USF)=0,0
Exp/Cntr=0.3,0.1

Type RM Length L Ch R = 1 ,29498   ,337.7,336.6,339.3
XS GIS Cut Line= 3
2209064.13603921639542.8872286042209316.95039924639667.341096786
2209375.54975421639876.066418312
#Sta/Elev= 30
       0 2131.93    22.7 2125.65    35.7 2120.58    71.4 2110.75   103.3 2109.27
   115.3 2105.17   124.9  2108.4   129.3 2108.73   138.3 2107.88   151.1 2104.45
     175 2106.83     193 2104.82   213.5 2105.59   227.4  2101.5   231.9 2101.22
   263.1 2099.82   300.3 2099.81   304.5 2098.59   315.1 2091.22   350.2 2089.48
   362.6 2091.17   386.5 2093.15   395.9 2096.18   404.2 2100.55   431.9 2102.36
   445.7 2109.87   458.2 2119.03   466.5 2123.11     479 2125.91   498.6 2132.58
#Mann= 3 ,-1,0
       0      .1       0   315.1    .045       0   362.6      .1       0
Bank Sta=315.1,362.6
XS Rating Curve= 0 ,0
Exp/Cntr(USF)=0,0
Exp/Cntr=0.3,0.1

Type RM Length L Ch R = 1 ,29161   ,314.2,312,303.3
XS GIS Cut Line= 3
2208948.97125693639568.4364679132209051.44992714639972.550469295
2209097.85536271640026.690144121
#Sta/Elev= 30
       0 2141.39       9 2141.09    13.1 2140.25    29.7 2128.49    59.2 2119.16
    78.1 2114.14   108.1  2110.5   121.8 2107.79   128.7  2105.6   144.8 2098.03
   149.3 2096.89   198.8 2096.29   223.8 2097.11   231.9 2095.16   240.1 2090.79
   244.2 2089.91   253.4 2089.63  269.392087.185   293.8 2086.25  319.632087.224
     335 2091.13   355.7 2093.55   372.2 2096.95   391.7 2097.82   408.1 2097.62
   413.4 2098.36   433.5 2103.67   460.4 2109.45   471.8 2113.01   488.2  2119.8
#Mann= 6 ,-1,0
       0     .06       0      60      .1       0     170     .06       0
     180      .1       0  269.39    .045       0  319.63      .1       0
Bank Sta=269.39,319.63
XS Rating Curve= 0 ,0
Exp/Cntr(USF)=0,0
Exp/Cntr=0.3,0.1

Type RM Length L Ch R = 1 ,28849   ,127.8,123.8,117.5
XS GIS Cut Line= 2
2208700.60170309639895.2761244572208876.34675027640142.897089016
#Sta/Elev= 30
       0 2112.93    13.1 2112.57    18.3 2110.81      24 2106.89    26.9 2104.51
    29.7 2101.47    31.8 2098.96    36.7  2090.8    38.4 2088.61    41.2 2085.88
    46.5 2084.35    54.6 2083.17    58.4 2081.96    61.3 2081.04    66.1 2080.73
    78.5 2081.06   85.542081.962    92.9 2083.61   107.2 2084.92     125 2090.25
   134.8 2091.84   139.7 2092.04   149.5 2091.18   158.8 2088.44   170.3 2092.11
   178.9 2093.31   242.7 2093.68   253.5 2094.36   289.5 2094.64   303.6 2095.66
#Mann= 4 ,-1,0
       0      .1       0      40     .06       0    58.4    .045       0
   85.54     .06       0
#XS Ineff= 2 , 0
                          146.31         2096.76
Permanent Ineff=
       F       F
Bank Sta=58.4,85.54
XS Rating Curve= 0 ,0
Exp/Cntr(USF)=0,0
Exp/Cntr=0.3,0.1

Type RM Length L Ch R = 1 ,28725   ,45.4,44.4,43.1
XS GIS Cut Line= 3
 2208584.3322747639982.4745046252208740.80359542640106.391389488
 2208822.7147566640145.246683894
#Sta/Elev= 30
       0 2136.63     7.5 2130.64    16.1 2124.29    30.1 2112.59    35.5 2106.83
    38.8 2102.92    40.6 2101.29      43 2100.35    55.9 2099.75    58.8 2098.27
    61.6 2096.26    66.1 2089.94    71.2 2083.92    74.32082.234    76.3 2081.42
    81.4  2080.7    91.6 2080.47   123.52081.735   127.4 2081.92   132.5 2082.93
   135.6 2084.68   139.7 2087.57   142.7 2089.16   147.8 2090.14   155.6 2090.12
   175.5 2092.41   204.2 2093.59   228.2 2095.42   256.5 2096.42   290.3    2097
#Mann= 4 ,-1,0
       0      .1       0      70     .06       0    74.3    .045       0
   123.5     .06       0
Bank Sta=74.3,123.5
XS Rating Curve= 0 ,0
Exp/Cntr(USF)=0,0
Exp/Cntr=0.3,0.1

Type RM Length L Ch R = 1 ,28681   ,47.3,48.2,47.9
XS GIS Cut Line= 3
2208559.56891943640025.1393576082208682.20108359640112.532394136
2208806.24281285640175.962823875
#Sta/Elev= 30
       0 2128.09    10.6  2119.5    13.9 2115.76    20.5 2106.57    23.4 2103.05
    25.3 2100.89    29.1 2097.61    30.2 2096.97    34.5 2096.14    43.5 2095.84
      55 2094.71    57.8 2092.84    59.7 2090.97    64.6    2085    66.4 2083.57
   68.972082.087      75 2080.84    95.1 2080.64   118.6 2081.51   123.5 2082.09
   129.5  2083.3   135.3 2085.92   149.6  2091.4   155.5 2091.99   160.8 2091.84
   202.2 2092.38   229.2 2094.81   256.1 2094.78   271.4 2093.95   289.9 2093.77
#Mann= 3 ,-1,0
       0     .06       0   68.97    .045       0   123.5     .06       0
Bank Sta=68.97,123.5
XS Rating Curve= 0 ,0
Exp/Cntr(USF)=0,0
Exp/Cntr=0.3,0.1

Type RM Length L Ch R = 1 ,28633   ,59,60,60.8
XS GIS Cut Line= 3
2208533.49196498640064.6071805562208656.12412914640152.000217085
2208780.16585841640215.430646823
#Sta/Elev= 30
       0 2111.51     8.2 2104.26    13.1 2100.32    19.5 2096.91    22.4 2095.96
    25.3 2095.51    42.5 2094.53    45.4 2093.79    59.7 2086.81    68.3 2081.93
    72.1 2080.38      77 2080.13   106.4 2080.44   111.3 2080.87  114.382081.977
   118.2  2083.8   121.2 2085.74   126.1 2089.44   128.5 2090.73     131 2091.53
   135.9 2091.99   154.5 2092.14   164.1 2092.63   195.6 2090.75   200.1 2091.18
     209 2093.57   216.9 2094.74   240.5  2095.3   258.5 2094.78   289.9 2092.35
#Mann= 4 ,-1,0
       0     .06       0    68.3    .045       0  114.38      .1       0
  200.59     .06       0
Bank Sta=68.3,114.38
XS Rating Curve= 0 ,0
Exp/Cntr(USF)=0,0
Exp/Cntr=0.3,0.1

Type RM Length L Ch R = 1 ,28573   ,141.6,134.9,128.5
XS GIS Cut Line= 3
2208487.71911023640096.9401016592208704.04858719640271.263854941
2208761.04077009640274.759505944
#Sta/Elev= 30
       0 2118.98    11.9 2112.23      16 2108.96    26.3 2099.02    31.4 2096.94
    46.8 2095.98      52 2095.09    57.1 2091.69    62.2  2085.6    64.1 2083.95
    68.8 2081.74    72.5 2080.88    77.6 2080.33   108.8  2080.6   123.9 2080.17
   128.5 2080.25   131.4 2080.92   134.3 2082.25   139.9 2088.03   142.7 2090.04
   145.6 2091.27   151.3 2092.02   160.2 2092.36   185.3 2090.63   236.9 2089.78
   247.2 2090.64   262.6 2094.11   274.5 2094.84     298 2094.35   334.9 2091.83
#Mann= 6 ,-1,0
       0      .1       0      20     .06       0    72.5    .045       0
   131.4     .06       0     150      .1       0     200     .05       0
Bank Sta=72.5,131.4
XS Rating Curve= 0 ,0
Exp/Cntr(USF)=0,0
Exp/Cntr=0.3,0.1

Type RM Length L Ch R = 1 ,28438   ,191.2,191.5,176
XS GIS Cut Line= 3
2208405.09909354640232.2595637082208693.97292994640348.853220566
2208736.14279842640353.010274036
#Sta/Elev= 30
       0 2113.22     3.3 2110.24     7.6 2107.39    11.9  2106.5    24.6 2106.04
    29.2 2104.09    33.5 2100.71    42.1 2092.15    50.8 2085.09    55.1 2082.81
   62.932080.669    72.3 2079.44    89.6 2078.63    95.3 2078.84   107.6 2080.65
   115.5  2082.2   119.8 2084.32     126 2088.69   128.4 2089.79   132.7  2090.3
     150 2090.79   205.9 2088.81   236.2 2090.23   244.9 2089.82   253.5  2088.3
   261.2 2087.86   275.1 2088.83   285.8  2091.9   292.3 2092.84   353.9 2091.94
#Mann= 7 ,-1,0
       0     .06       0   62.93    .045       0   107.6     .06       0
     110      .1       0     210     .05       0     230      .1       0
  321.52     .05       0
Bank Sta=62.93,107.6
XS Rating Curve= 0 ,0
Exp/Cntr(USF)=0,0
Exp/Cntr=0.3,0.1

Type RM Length L Ch R = 1 ,28247   ,239.7,235.2,225.7
XS GIS Cut Line= 3
2208274.06370902640409.1527622282208659.38946098640464.481588151
2208718.35853295640466.829573079
#Sta/Elev= 30
       0 2149.02       9 2143.77    22.3 2134.67    38.5 2129.07    50.6 2116.63
    54.7 2113.34    58.7 2112.34    74.9 2111.67    78.9 2110.24      83 2106.62
    95.1 2092.65    99.1 2087.28   103.2  2083.1   107.2 2080.95   111.4 2079.84
   123.4 2077.94   143.2 2078.25   167.8 2079.61   175.9 2082.48     184 2086.92
   192.1 2088.53   305.8 2086.75   325.4 2088.73   341.6 2088.18   357.7 2086.68
   377.9 2088.05   390.1 2090.92   398.1 2091.98   421.5 2090.36   448.3 2090.12
#Mann= 5 ,-1,0
       0      .1       0   111.4    .045       0   167.8     .06       0
     230      .1       0  429.28     .05       0
Bank Sta=111.4,167.8
XS Rating Curve= 0 ,0
Exp/Cntr(USF)=0,0
Exp/Cntr=0.3,0.1

Type RM Length L Ch R = 1 ,28011   ,300.1,292.5,287
XS GIS Cut Line= 2
2208294.57585966640678.267361087 2208753.9270639640605.546843788
#Sta/Elev= 30
       0 2142.07     5.7 2138.62    17.8 2133.92      30 2126.79      34 2123.44
    42.1    2115    46.2 2113.41    66.4 2112.51    70.5 2111.11    74.5 2108.01
    90.7 2090.98   100.2 2082.43   103.7 2079.64108.70992077.337   127.2 2075.88
   139.3 2077.29   147.4 2077.67   159.7 2076.76   163.6  2077.4   175.8 2082.05
   187.9 2085.26   208.2 2087.36   232.5 2086.63   248.7 2087.09   256.8 2086.23
     277 2085.83   366.3 2087.47   398.5 2084.66   426.8 2086.14   465.1  2085.7
#Mann= 5 ,-1,0
       0      .1       0108.7099    .045       0   139.3     .06       0
     210      .1       0     410     .05       0
#XS Ineff= 2 , 0
                          576.46         2091.28
Permanent Ineff=
       F       F
Bank Sta=108.7099,139.3
XS Rating Curve= 0 ,0
Exp/Cntr(USF)=0,0
Exp/Cntr=0.3,0.1

Type RM Length L Ch R = 1 ,27719   ,214.1,208.4,205.6
XS GIS Cut Line= 2
2208414.36180332640990.105434425 2208791.2740214640762.048379973
#Sta/Elev= 30
       0 2126.94    30.2 2116.97    40.4 2110.45    45.7  2107.9    48.9  2107.4
    67.6 2107.47    71.9 2105.96    79.1 2100.95    86.3 2093.49   103.9 2076.74
   109.6 2074.33   125.4    2073   137.7 2073.77   147.1 2073.66   150.5 2074.39
   159.3 2078.32   165.8 2079.85   171.8 2080.03   200.1 2078.25   217.2 2079.94
   231.2 2083.82   235.9 2084.27   264.1 2083.36   287.3 2083.57   304.9 2082.54
   325.3  2083.1   360.3 2082.81   383.6  2084.6   395.9 2084.92   440.5 2084.34
#Mann= 5 ,-1,0
       0      .1       0   109.6    .045       0   150.5     .06       0
     170      .1       0     360     .05       0
Bank Sta=109.6,150.5
XS Rating Curve= 0 ,0
Exp/Cntr(USF)=0,0
Exp/Cntr=0.3,0.1

Type RM Length L Ch R = 1 ,27510   ,474.5,440.2,422.7
XS GIS Cut Line= 2
2208557.15805679641177.1735356322208944.21870449640817.179602947
#Sta/Elev= 30
       0  2104.3    50.2 2103.14    64.6 2102.55    70.1 2101.85    75.1 2098.94
    84.2 2092.14    95.5 2080.14    99.8 2076.48     104 2074.67   113.4 2073.68
     121 2072.91   135.2 2072.63   152.7 2072.96   158.6 2073.75   166.3 2076.38
   173.5 2077.39   193.8 2077.33   208.7  2075.8   217.2  2075.9   234.9 2077.84
   245.5 2081.08   251.2  2081.8   270.2 2081.24   299.1  2081.7   337.3 2081.51
   370.1 2080.59   397.4 2078.95   452.2 2077.62   517.2 2079.66   528.6 2081.09
#Mann= 5 ,-1,0
       0     .06       0   113.4    .045       0   158.6     .06       0
     200      .1       0     470     .05       0
#XS Ineff= 2 , 0
                          338.83         2083.59
Permanent Ineff=
       F       F
Bank Sta=113.4,158.6
XS Rating Curve= 0 ,0
Exp/Cntr(USF)=0,0
Exp/Cntr=0.3,0.1

Type RM Length L Ch R = 1 ,27070   ,60.3,67,54.5
XS GIS Cut Line= 6
2208930.67280368641442.3538296242209012.52587095641443.594027613
 2209029.2685438641369.1821482812209035.46953374641282.988388055
2209009.42537598641132.3043324092208970.35913933640974.179088829
#Sta/Elev= 30
       0 2092.79    33.5 2090.64    53.5 2088.34    61.5 2085.61    69.5 2079.94
    73.5  2077.7    77.5 2076.49   104.8 2076.73   121.2 2080.44   129.4 2078.75
   141.7 2078.39   158.1 2072.31  168.692069.802   174.2 2068.52   189.6 2068.06
   202.3 2069.28   239.4 2069.11   254.5 2069.77   258.6 2071.26   270.7  2077.7
   274.8 2078.82   278.9    2079     291  2077.9   319.5 2078.14   376.3 2076.34
   429.5 2077.63   450.1 2078.75   540.8 2078.83   552.8 2079.57   560.3  2079.1
#Mann= 3 ,-1,0
       0      .1       0  168.69    .045       0   254.5      .1       0
Bank Sta=168.69,254.5
XS Rating Curve= 0 ,0
Exp/Cntr(USF)=0,0
Exp/Cntr=0.3,0.1

Type RM Length L Ch R = 1 ,27003   ,129.1,164.7,205.1
XS GIS Cut Line= 6
2208983.07116871641461.2668489542209064.92423598641462.507046943
2209081.66690883641388.0951676112209087.86789877641301.901407385
2209050.66195911641148.7369557612209009.11532648640980.070029276
#Sta/Elev= 30
       0 2088.41    17.1  2081.6    25.1 2076.45    45.1 2072.41    57.1 2072.08
    69.1 2070.57    77.1 2068.78   100.5 2069.02   112.5 2070.18   120.1 2071.63
   124.2 2071.71   136.5 2071.19   148.8 2069.12   155.52069.312   165.1 2068.39
   193.1 2069.12   237.3 2068.93   248.2 2068.46   256.8 2069.21     270 2070.25
   294.7 2071.14   317.8 2073.79     340 2074.07   350.9 2074.72   429.3 2074.34
   488.2 2074.78   517.1  2075.6   554.1 2075.84   565.8 2076.87   575.9  2076.5
#Mann= 4 ,-1,0
       0      .1       0   155.5    .045       0   256.8      .1       0
  552.17     .05       0
Bank Sta=155.5,256.8
XS Rating Curve= 0 ,0
Exp/Cntr(USF)=0,0
Exp/Cntr=0.3,0.1

Type RM Length L Ch R = 1 ,26839   ,206.6,219.5,240.8
XS GIS Cut Line= 3
2208957.76991507641497.9450152232209098.06800938641525.609428185
2209449.80125989641282.557800021
#Sta/Elev= 30
       0 2091.44    18.8 2089.06    38.9 2080.45    47.3    2074    51.4 2072.13
    67.7 2071.94    79.9 2068.58   103.6 2068.27   112.5 2071.38   141.1 2074.09
   150.6 2077.41   169.9 2072.29   190.8 2072.08   213.6 2073.83   223.4 2069.18
   242.8 2067.68   256.3 2067.02   282.8 2067.58   286.6 2068.56   296.3 2074.17
   301.1 2074.72   343.2 2073.15   359.5 2070.47   374.1  2074.9   389.2 2082.65
   397.8 2085.94   408.1 2088.25   481.5 2094.03   524.8 2099.46   570.5 2103.88
#Mann= 3 ,-1,0
       0      .1       0   242.8    .045       0   282.8      .1       0
#XS Ineff= 2 ,-1
  150.42  209.58 2079.02  302.54   570.5 2080.41
Permanent Ineff=
       F       F
Bank Sta=242.8,282.8
XS Rating Curve= 0 ,0
Exp/Cntr(USF)=0,0
Exp/Cntr=0.3,0.1

Type RM Length L Ch R = 1 ,26619   ,343.9,350.6,365.8
XS GIS Cut Line= 2
2208925.93723392641574.2173363022209426.72922606641682.496685955
#Sta/Elev= 30
       0 2088.32    14.5 2085.62    18.7 2083.88    27.9 2078.94    39.1 2070.42
    43.2 2069.65    59.6 2069.93      75 2065.38    91.9 2063.83    96.4 2064.33
   112.8 2071.17     121 2072.19   137.3 2071.09   170.1 2071.74   186.4 2069.92
   194.6 2066.38     211 2067.88   219.2 2069.85   243.7  2070.9     256 2073.54
   321.5 2072.06   337.9 2070.79   350.1 2066.45   362.4  2065.2  393.132066.476
   403.3 2069.34   452.5 2097.24   468.8 2100.31   497.5  2102.8   512.4 2105.21
#Mann= 3 ,-1,0
       0      .1       0   350.1    .045       0  393.13      .1       0
Bank Sta=350.1,393.13
XS Rating Curve= 0 ,0
Exp/Cntr(USF)=0,0
Exp/Cntr=0.3,0.1

Type RM Length L Ch R = 1 ,26269   ,384.4,389,402.4
XS GIS Cut Line= 2
2208871.79755909  641599.35361392209223.70544546642063.407969554
#Sta/Elev= 30
       0 2087.62    27.3 2084.45      53 2074.78    64.4 2068.11    81.5 2067.78
    92.9 2063.16    97.7 2062.63   112.9 2063.34   124.3 2066.41   132.8 2066.91
   159.5 2063.93     188 2066.46     210  2063.8   227.1 2068.46   288.4  2070.2
   338.6 2067.38   404.4 2069.28   413.9 2068.46     429 2064.89   444.2 2064.11
   452.7 2062.29   459.1 2061.66  481.982062.259   486.9 2064.35   495.5 2070.36
   509.8 2081.55   526.8 2096.96   546.9 2110.34   559.5 2115.01   582.4  2115.7
#Mann= 3 ,-1,0
       0      .1       0   452.7    .045       0  481.98      .1       0
Bank Sta=452.7,481.98
XS Rating Curve= 0 ,0
Exp/Cntr(USF)=0,0
Exp/Cntr=0.3,0.1

Type RM Length L Ch R = 1 ,25880   ,401,408.9,414.3
XS GIS Cut Line= 2
2208768.49052934641611.3566580732208777.13368236642272.557864187
#Sta/Elev= 30
       0 2085.68    45.8 2079.75    81.8 2072.36   101.8 2064.18   137.8 2065.24
   153.8 2064.34   169.8 2066.31   173.8 2065.73   185.8 2060.33   213.8 2059.19
   229.8 2062.83   257.5 2064.56   301.8 2065.53   329.2  2064.8   357.9 2066.14
   369.9  2064.3   377.9 2059.44   383.2 2057.81   389.9 2057.03   417.9 2057.87
   425.9 2058.86   437.9 2062.95   465.9 2061.04   545.9 2062.99   565.9 2059.71
     578 2065.18   617.9 2066.23   625.9 2068.61   645.1 2083.02   661.3 2090.46
#Mann= 3 ,-1,0
       0      .1       0   383.2    .045       0   417.9      .1       0
Bank Sta=383.2,417.9
XS Rating Curve= 0 ,0
Exp/Cntr(USF)=0,0
Exp/Cntr=0.3,0.1

Type RM Length L Ch R = 1 ,25471   ,492,497.8,499
XS GIS Cut Line= 2
2208510.22187364 641554.881738152208299.46385378642173.620879022
#Sta/Elev= 30
       0 2068.06    85.4 2065.46    91.7 2064.52   108.1 2058.58     125 2057.19
     163 2059.28   196.8 2058.57   218.3 2060.18     256 2059.16   272.9 2060.36
   281.3 2058.13   289.8 2053.23   302.5 2051.72   310.9 2051.99   324.9 2055.18
   340.5 2056.49   391.1 2056.44  402.652052.569   438.4 2051.72   446.1 2052.58
   466.8 2064.11   473.1 2066.44   509.5  2069.3   522.2 2073.24   543.3 2076.33
   567.6 2075.06   583.4 2078.79   602.5  2080.2   636.3 2088.28   653.6 2089.66
#Mann= 3 ,-1,0
       0      .1       0  402.65    .045       0   446.1      .1       0
#XS Ineff= 2 , 0
          158.64 2064.68
Permanent Ineff=
       F       F
Bank Sta=402.65,446.1
XS Rating Curve= 0 ,0
Exp/Cntr(USF)=0,0
Exp/Cntr=0.3,0.1

Type RM Length L Ch R = 1 ,24973   ,428.9,420.7,397.1
XS GIS Cut Line= 3
2208111.90855171641394.3962734862207822.04727658641969.863872266
2207922.24699266 642338.24518137
#Sta/Elev= 30
       0 2072.37    47.9 2068.36    74.8 2062.96    92.7 2063.53   115.1 2056.09
     124 2054.44   177.8 2054.83   222.3 2050.56   284.8 2052.88   301.7 2050.54
   323.6 2050.55   337.3 2052.25   361.4 2048.02  378.962046.577   392.8 2044.78
   406.2 2045.77   421.8 2044.91   430.8  2046.6     451 2055.78     460 2056.54
   482.3 2055.04   681.4 2050.07   701.7  2051.7   888.2 2049.98   896.6 2052.04
   917.2 2061.43   929.7 2064.72   942.1 2071.17     967 2076.94  1026.1 2098.56
#Mann= 3 ,-1,0
       0      .1       0  378.96    .045       0   430.8      .1       0
#XS Ineff= 2 , 0
          270.63 2058.51  592.74         2059.79
Permanent Ineff=
       F       F
Bank Sta=378.96,430.8
XS Rating Curve= 0 ,0
Exp/Cntr(USF)=0,0
Exp/Cntr=0.3,0.1

Type RM Length L Ch R = 1 ,24552   ,410.4,396.6,361.3
XS GIS Cut Line= 3
2207574.49503686 641392.241979592207587.61536346642048.991124483
2207764.71013344642354.998782775
#Sta/Elev= 30
       0 2100.79    12.9 2099.91    27.8 2093.31    49.6 2077.33      81 2057.37
      89 2049.23    92.8 2047.04     117  2045.4127.14722040.272     149 2038.96
 188.2812040.424     213 2047.09     225 2046.92     241 2050.39     261 2050.13
     277  2051.9     341 2049.07     417 2048.85     445 2050.59     485 2050.69
     521 2049.13   605.1 2049.46   712.6 2047.62   748.2 2045.35   786.2  2047.1
   809.6 2042.53   837.3 2046.85   925.1 2048.27   988.2 2066.12  1010.4 2075.02
#Mann= 4 ,-1,0
       0     .06       0      10      .1       0127.1472    .045       0
 188.281      .1       0
#XS Ineff= 2 , 0
                          660.07         2057.66
Permanent Ineff=
       F       F
Bank Sta=127.1472,188.281
XS Rating Curve= 0 ,0
Exp/Cntr(USF)=0,0
Exp/Cntr=0.3,0.1

Type RM Length L Ch R = 1 ,24156   ,311.1,312.2,307.4
XS GIS Cut Line= 3
2207106.23027613641620.458844054 2207416.4669072641920.815327638
2207554.78897201642399.014465977
#Sta/Elev= 30
       0 2092.74      24 2084.63    44.3 2083.97    58.5 2085.05    78.3 2080.15
   136.3 2073.55   162.1 2068.53   191.4 2065.44   199.9 2061.02     214 2046.81
   219.7 2043.11     231 2042.32   253.2 2037.69   288.6  2036.3   303.4 2037.67
   325.6 2043.41   372.5 2046.36   412.1 2046.56     490 2044.01   541.7 2047.38
   693.5 2044.83   736.2 2045.47   790.3 2043.59   816.2 2044.28   823.6 2043.58
   836.1 2039.07     842 2038.92   848.5 2040.25   874.3 2051.86   929.6 2068.99
#Mann= 3 ,-1,0
       0      .1       0   253.2    .045       0   303.4      .1       0
#XS Ineff= 2 , 0
                          811.83         2049.41
Permanent Ineff=
       F       F
Bank Sta=253.2,303.4
XS Rating Curve= 0 ,0
Exp/Cntr(USF)=0,0
Exp/Cntr=0.3,0.1

Type RM Length L Ch R = 1 ,23843   ,238.8,239.9,241.3
XS GIS Cut Line= 2
 2206843.6265196641822.5113486242207523.85292154642395.046632183
#Sta/Elev= 30
       0 2099.19    26.9 2090.84    66.3 2082.58   105.3 2068.01     147 2056.75
   209.8 2049.77   225.5  2045.3   251.7 2046.23   277.5 2039.89   298.7 2039.97
   311.7 2034.38   325.9 2034.24   340.6  2037.2   361.5 2035.37   402.6 2033.75
  409.782035.319     419 2041.61   433.8 2043.32   617.7 2041.63   635.3 2038.54
   658.1 2044.34   699.9 2042.14   758.8 2044.55     785    2042   800.6 2042.84
   814.2 2038.71   825.6 2038.66   836.5  2041.3   868.1 2057.15   889.1 2065.02
#Mann= 3 ,-1,0
       0      .1       0   361.5    .045       0  409.78      .1       0
#XS Ineff= 2 , 0
                          572.96         2045.59
Permanent Ineff=
       F       F
Bank Sta=361.5,409.78
XS Rating Curve= 0 ,0
Exp/Cntr(USF)=0,0
Exp/Cntr=0.3,0.1

Type RM Length L Ch R = 1 ,23603   ,229.8,231,232.7
XS GIS Cut Line= 2
2206738.68878964641976.1441535622207278.14484239642580.809179726
#Sta/Elev= 30
       0 2081.79    14.2 2074.23    44.3 2061.63    75.4 2053.28   167.6 2041.78
   183.1 2037.56   205.1 2039.08   245.4 2037.61   256.8 2038.53   306.9 2034.58
     323 2030.71   330.4 2030.32   355.2 2032.37   365.9 2031.18   389.9 2031.36
   408.8 2040.54   422.8 2041.77   464.9 2040.39   505.3 2037.28   526.7 2039.07
     561    2038     625 2039.57   671.5 2038.82   698.7 2035.22   719.7 2035.49
   730.4 2040.17   741.1 2048.86   758.2 2059.98   777.3 2075.76   810.3 2082.82
#Mann= 3 ,-1,0
       0      .1       0   365.9    .045       0   389.9      .1       0
#XS Ineff= 2 , 0
                           629.3         2043.62
Permanent Ineff=
       F       F
Bank Sta=365.9,389.9
XS Rating Curve= 0 ,0
Exp/Cntr(USF)=0,0
Exp/Cntr=0.3,0.1

Type RM Length L Ch R = 1 ,23372   ,428.6,436.2,444.5
XS GIS Cut Line= 2
2206584.07127076642104.7421861562207032.67784273642694.152280723
#Sta/Elev= 30
       0 2074.84    23.2 2060.32    34.6 2056.53    51.8 2046.41    68.9 2040.69
      81 2038.76   121.2 2038.94   163.1 2033.92   186.5 2035.65   211.7 2034.72
   251.9 2037.51   257.3 2036.92   265.8 2033.64     277 2035.22   302.9 2032.02
   332.3  2032.2  355.742028.269   396.4  2027.1  405.232028.339     420 2036.17
   425.7 2037.42   478.1 2037.09   498.2 2033.94   582.7 2036.18   605.5  2033.2
   628.9 2033.24     639 2037.21   684.2 2067.27   699.7 2075.62   740.7 2089.07
#Mann= 3 ,-1,0
       0      .1       0  355.74    .045       0  405.23      .1       0
#XS Ineff= 2 , 0
          278.11 2044.57  475.25         2044.95
Permanent Ineff=
       F       F
Bank Sta=355.74,405.23
XS Rating Curve= 0 ,0
Exp/Cntr(USF)=0,0
Exp/Cntr=0.3,0.1

Type RM Length L Ch R = 1 ,22936   ,479.9,475.3,463.4
XS GIS Cut Line= 2
 2206279.5427219642245.5457087472206561.14976708642880.798810669
#Sta/Elev= 30
       0 2104.97    43.4 2080.84      74 2065.83   117.7 2039.24   135.2  2031.9
   152.7 2030.45   165.9 2031.34   187.7 2030.71   212.4  2032.2   224.5 2031.32
   279.6  2032.6   292.8 2031.75   318.5 2032.35   336.5 2030.31     347 2031.55
   357.9 2030.24   373.1 2030.24   393.4 2027.53     424 2028.21  434.922025.892
   442.8 2025.43   502.8 2025.91   533.4 2029.83   554.3 2041.14   563.9 2043.91
   590.3 2047.28     634 2055.29     652 2057.35   677.8 2062.07   694.9  2066.9
#Mann= 3 ,-1,0
       0      .1       0  434.92    .045       0   502.8      .1       0
#XS Ineff= 2 , 0
          313.42 2044.47
Permanent Ineff=
       F       F
Bank Sta=434.92,502.8
XS Rating Curve= 0 ,0
Exp/Cntr(USF)=0,0
Exp/Cntr=0.3,0.1

Type RM Length L Ch R = 1 ,22461   ,348.9,333.1,319.7
XS GIS Cut Line= 3
2205956.70563462642239.1075177372206023.56362094642845.744378826
 2206264.8374376 643117.64293748
#Sta/Elev= 30
       0 2115.53    54.4 2089.32    74.5 2073.15    98.7 2050.31   110.7 2046.45
   126.8 2036.27     147 2032.06   171.1 2028.89   227.4 2029.57   307.9 2027.38
   344.1  2029.8   460.8 2026.75   521.2 2027.36   577.5 2025.87   609.7 2027.39
   625.6 2026.47633.07042021.632   638.7 2019.97   665.5 2019.81685.58982021.408
     701 2024.14   727.2 2024.34   748.6 2027.01   810.1 2025.58   822.9 2020.93
   831.4 2020.85   844.9 2024.64   860.9 2037.49     922 2045.78   973.8  2057.8
#Mann= 3 ,-1,0
       0      .1       0633.0704    .045       0685.5898      .1       0
#XS Ineff= 2 , 0
           606.2 2039.96
Permanent Ineff=
       F       F
Bank Sta=633.0704,685.5898
XS Rating Curve= 0 ,0
Exp/Cntr(USF)=0,0
Exp/Cntr=0.3,0.1

Type RM Length L Ch R = 1 ,22128   ,170.8,168.4,172.9
XS GIS Cut Line= 3
2205835.64330939642205.3635752452205772.41036547643114.337143989
2206167.61626493643268.467444776
#Sta/Elev= 30
       0 2106.67    19.9 2096.48      72 2074.65      96 2056.58   124.1  2040.6
   132.1 2037.63   152.2 2034.58   192.3  2032.7   228.4 2033.82   360.7 2031.39
   440.9 2025.86   545.1 2024.93   573.5    2027   709.5 2021.79   777.7 2023.24
   805.8 2020.21   837.8 2022.16   947.2 2023.48   976.1 2018.77  1048.3 2018.72
  1086.2 2021.24  1104.1 2017.36  1112.7 2019.48  1123.2 2029.05  1134.2 2032.46
  1207.2 2039.08  1258.7  2047.9  1302.4 2060.05  1327.1 2069.07  1335.4 2069.26
#Mann= 3 ,-1,0
       0      .1       0   976.1    .045       0  1048.3      .1       0
#XS Ineff= 2 , 0
          905.52 2025.96
Permanent Ineff=
       F       F
Bank Sta=976.1,1048.3
XS Rating Curve= 0 ,0
Exp/Cntr(USF)=0,0
Exp/Cntr=0.3,0.1
