HEC-RAS study LFBUCKRV.prj: LFBUCKRV

--- LFBUCKRV.g01 (geometry) --- (continued)

Type RM Length L Ch R = 1 ,21959   ,320.2,320,319.4
XS GIS Cut Line= 2
2205431.56443362643173.9812753442206031.00203177643386.369422007
#Sta/Elev= 30
       0 2058.38    13.4  2043.8    17.6 2039.91    34.6 2026.71    38.8 2023.82
    43.7 2021.76    55.8    2021   105.4 2021.97   119.5 2020.54   132.2 2015.57
   157.7  2014.2   189.2 2018.12   208.6 2018.69   217.1 2019.85   237.1 2018.59
   301.9 2020.73   323.2  2020.1   361.4 2023.21   392.8 2015.88   475.5 2014.98
   480.2 2015.08  481.89 2015.88   491.8 2020.35   497.2 2023.72   509.9 2035.23
   514.1 2037.88   528.1 2040.74   556.6 2044.47   582.7 2049.18     636 2063.68
#Mann= 3 ,-1,0
       0      .1       0   392.8    .045       0  481.89      .1       0
#XS Ineff= 2 , 0
          328.41 2031.84
Permanent Ineff=
       F       F
Bank Sta=392.8,481.89
XS Rating Curve= 0 ,0
Exp/Cntr(USF)=0,0
Exp/Cntr=0.3,0.1

Type RM Length L Ch R = 1 ,21639   ,405.1,410.2,410.6
XS GIS Cut Line= 2
2205312.48998752643458.0720804662205893.25679533643676.578404194
#Sta/Elev= 30
       0 2064.96     8.2 2059.22    25.3  2049.6    45.6 2030.73    63.8  2015.8
    76.6 2011.18    89.4 2010.57   102.2 2012.82   119.3    2013   149.2    2017
   162.1 2015.94   187.7 2016.03   226.2 2019.69   268.9  2018.7   320.2 2019.39
   337.3 2017.77   353.1 2019.24   367.2 2018.56     381 2015.36   397.1 2015.32
  434.28  2012.3   465.5 2011.38   489.7  2012.3   508.3 2016.77   533.9 2035.46
     556 2049.14   576.7 2064.16   589.4 2075.07   610.8 2086.06   620.5  2088.9
#Mann= 3 ,-1,0
       0      .1       0  434.28    .045       0   489.7      .1       0
#XS Ineff= 2 , 0
          292.18 2034.93
Permanent Ineff=
       F       F
Bank Sta=434.28,489.7
XS Rating Curve= 0 ,0
Exp/Cntr(USF)=0,0
Exp/Cntr=0.3,0.1

Type RM Length L Ch R = 1 ,21229   ,437.4,436.4,433.8
XS GIS Cut Line= 3
2205201.32010352643860.5837294382205409.34373576643908.183939396
2205654.39783329644016.645841728
#Sta/Elev= 30
       0 2052.48    15.2 2046.43    23.4 2041.68    31.7 2034.04      44 2020.95
    49.6 2016.78    56.3 2013.22    68.6 2010.18      85 2011.02    97.3 2007.96
   117.8 2007.93   129.8 2009.87   142.4 2014.34   150.7 2013.67     163 2014.94
   175.3 2014.02   187.6 2015.93   229.6 2016.22   251.5 2013.94   264.6 2014.41
  298.33 2008.15   324.6 2007.53   342.6 2008.15   356.5 2009.03   378.3 2013.23
   391.5 2023.52   407.3 2037.43   416.4 2043.25   448.3  2058.3   481.4 2070.52
#Mann= 3 ,-1,0
       0      .1       0  298.33    .045       0   342.6      .1       0
#XS Ineff= 2 , 0
          200.44 2029.41
Permanent Ineff=
       F       F
Bank Sta=298.33,342.6
XS Rating Curve= 0 ,0
Exp/Cntr(USF)=0,0
Exp/Cntr=0.3,0.1

Type RM Length L Ch R = 1 ,20793   ,363.6,371.8,386
XS GIS Cut Line= 2
2205026.53229085 644258.570231652205571.05093117644411.554040123
#Sta/Elev= 30
       0 2055.81    80.6 2031.65    93.1 2031.54   101.4 2028.17     118 2024.25
   130.5 2019.99   163.7 2016.49   192.8 2009.72   213.6 2009.81   226.1 2008.11
   242.7 2009.92   287.5 2002.97   292.5 2002.58   314.8 2002.95   334.1 2003.31
   350.7 2007.07     359 2007.63   367.3 2006.89   379.8 2003.91   395.9 2007.09
   404.7 2010.16   417.2 2009.25   433.8 2017.23   447.8 2028.54   454.3 2032.24
   479.5 2043.67   508.6 2053.66   525.2 2061.23   537.7 2065.33   565.6 2078.27
#Mann= 3 ,-1,0
       0      .1       0   287.5    .045       0   314.8      .1       0
Bank Sta=287.5,314.8
XS Rating Curve= 0 ,0
Exp/Cntr(USF)=0,0
Exp/Cntr=0.3,0.1

Type RM Length L Ch R = 1 ,20421   ,417.7,425,433.7
XS GIS Cut Line= 3
2204968.63622814644503.4184726512205462.76818092644794.646000377
 2205479.4779571644947.421096888
#Sta/Elev= 30
       0  2035.2    27.3 2023.01    42.9 2020.16    56.5 2014.72      74 2014.22
    87.7 2009.43   117.8 2009.66   129.5 2006.41   138.8 2007.81   217.1 2008.57
   231.6 2006.84   259.5 2006.89   296.6 2004.16   316.4 2006.56   338.4 2006.42
   361.6 2001.67   375.6 2000.43   392.4 1999.36   428.9 2000.36   444.6 2010.12
   454.5 2011.98   474.2 2019.56     487 2026.55   497.6 2025.63   519.5 2031.31
   561.3 2036.26   580.1 2037.96   608.3 2038.17   640.5 2045.64   727.3 2069.08
#Mann= 3 ,-1,0
       0      .1       0   375.6    .045       0   428.9      .1       0
#XS Ineff= 2 , 0
          199.66 2016.81
Permanent Ineff=
       F       F
Bank Sta=375.6,428.9
XS Rating Curve= 0 ,0
Exp/Cntr(USF)=0,0
Exp/Cntr=0.3,0.1

Type RM Length L Ch R = 1 ,19996   ,447.8,445.5,444.1
XS GIS Cut Line= 2
2204751.43300889644718.1629676852205279.29483845645290.496672993
#Sta/Elev= 30
       0 2056.12    19.6  2048.8    53.1 2037.16    84.8 2024.47   113.2 2014.29
   135.7 2003.82   138.5 2003.79     147 2004.98   161.9 2003.27   200.8 2004.01
   266.6 2003.66   325.4 2003.97     365 2002.25  395.391996.826   407.5 1995.85
   444.3 1995.85   449.9 1996.17   452.7 1996.87   466.9  2001.6   483.9 2008.35
   499.3 2013.08   510.2 2017.92     521 2020.29   580.9 2043.44     597 2047.99
   657.1 2069.62   695.2 2081.98   706.1 2084.49   727.3 2092.09   778.6 2107.92
#Mann= 3 ,-1,0
       0      .1       0  395.39    .045       0   452.7      .1       0
Bank Sta=395.39,452.7
XS Rating Curve= 0 ,0
Exp/Cntr(USF)=0,0
Exp/Cntr=0.3,0.1

Type RM Length L Ch R = 1 ,19551   ,506.1,524.4,539.1
XS GIS Cut Line= 2
2204461.44677883645085.0380392932204898.28807041 645512.33088735
#Sta/Elev= 30
       0 2009.87    16.2 2009.67    26.2 2007.51    52.9 2004.43    57.4 2003.35
    67.1 1998.62    80.3 1999.08    95.4 1996.52   104.5 1993.71   123.7 1995.86
     189 1996.61   328.3 1999.93   350.7 1999.11   366.3 1999.67   395.5 1993.46
   429.1 1992.75   446.1 1993.45   468.7 1996.21   480.1  2000.2   494.2 1999.47
   502.7 2000.68   507.4  2002.3     514  2007.6   518.6  2010.2   539.5 2011.97
   549.4 2017.11   556.4 2019.53   583.7 2026.59   591.3 2027.22   611.1 2031.38
#Mann= 3 ,-1,0
       0      .1       0   395.5    .045       0   446.1      .1       0
#XS Ineff= 1 ,-1
   327.4  363.19 2001.31
Permanent Ineff=
       F
Bank Sta=395.5,446.1
XS Rating Curve= 0 ,0
Exp/Cntr(USF)=0,0
Exp/Cntr=0.3,0.1

Type RM Length L Ch R = 1 ,19026   ,546.3,568.1,586.1
XS GIS Cut Line= 2
2204206.02591434645161.4255875492204406.54322852645918.139737459
#Sta/Elev= 30
       0 2014.91    34.3 2009.92    61.8 2003.95    99.1 2000.82   115.6 2000.84
   123.9 1998.97   135.7 1993.72   148.8 1994.72   169.4 1990.07   214.9 1990.19
   223.2 1992.37   264.6 1994.09     306 1994.26   326.7 1992.01   363.9 1995.28
   400.6 1995.91   479.8 1993.56  495.331990.539   529.4 1989.57   562.5 1990.56
   579.1 1995.73   616.3 1995.27   657.7 1998.14   670.1  2002.1   685.2 2012.61
   690.8 2014.74   736.3 2013.92   744.6 2017.28     758  2019.1   782.8 2026.12
#Mann= 3 ,-1,0
       0      .1       0  495.33    .045       0   562.5      .1       0
#XS Ineff= 2 , 0
                          590.87         1998.56
Permanent Ineff=
       F       F
Bank Sta=495.33,562.5
XS Rating Curve= 0 ,0
Exp/Cntr(USF)=0,0
Exp/Cntr=0.3,0.1

Type RM Length L Ch R = 1 ,18458   ,290.3,286.3,280.8
XS GIS Cut Line= 2
2203986.41171311645175.748252847 2203721.4424051645782.074417128
#Sta/Elev= 30
       0 2010.78    36.5 2007.49    53.9 2007.37    65.5 2005.28   158.7 1999.02
   167.4 1997.12   176.2 1991.43   180.5 1990.78   189.3 1991.41   202.4 1989.82
   267.8 1985.84   289.7 1987.84   307.1 1985.35   355.1 1987.97   385.5 1987.28
   400.7 1990.55   429.4 1987.77   443.3    1984   464.5 1983.26   491.9 1983.99
     504    1989   516.2 1991.12   528.3 1999.41   538.5 2003.93     583 2013.79
   595.2 2017.66   604.3  2018.9   630.2 2029.14   644.9 2037.33   661.7 2040.36
#Mann= 3 ,-1,0
       0      .1       0   443.3    .045       0   491.9      .1       0
Bank Sta=443.3,491.9
XS Rating Curve= 0 ,0
Exp/Cntr(USF)=0,0
Exp/Cntr=0.3,0.1

Type RM Length L Ch R = 1 ,18172   ,261.8,257.1,256
XS GIS Cut Line= 2
2203623.74855553645079.2376109992203485.02594954645708.026993281
#Sta/Elev= 30
       0 2010.82    18.4 2006.78    28.1 2003.28    42.9 2002.66    75.1 1996.53
   100.3 1994.46   120.8  1990.6   157.6 1986.18   206.8 1988.81   223.2 1986.73
   239.6 1987.62   251.9 1986.61   276.4 1989.16   296.9 1985.94   337.9  1987.6
   346.1  1986.1   358.4 1981.36   419.8 1983.84   434.2 1980.81     473 1980.04
   481.9 1980.83   489.4 1983.83   526.3  1986.9   530.4 1988.52   538.6 1994.86
   575.1 2017.58     600 2028.73   625.5 2038.05   636.9 2046.25   643.9 2047.48
#Mann= 3 ,-1,0
       0      .1       0   434.2    .045       0   481.9      .1       0
#XS Ineff= 2 , 0
          324.17  1993.6
Permanent Ineff=
       F       F
Bank Sta=434.2,481.9
XS Rating Curve= 0 ,0
Exp/Cntr(USF)=0,0
Exp/Cntr=0.3,0.1

Type RM Length L Ch R = 1 ,17915   ,232.3,253.7,293.1
XS GIS Cut Line= 3
2203346.30334356645053.3081519362203277.59027704645411.134687007
2203280.18322294645671.725750592
#Sta/Elev= 30
       0 2010.28    24.3 2009.78    48.7 2004.27    77.3 1984.63    81.3 1983.43
    97.6 1983.06   130.2  1988.1   207.6 1986.88     232 1988.85   244.3 1984.44
   256.5    1985   272.8 1983.27   301.3 1984.34   317.6  1983.4   350.7 1985.45
   382.4 1984.84   386.4 1984.03   398.4 1977.21   414.4 1976.67   430.4 1977.22
   462.4 1978.36   478.4 1981.75   494.4 1981.01   514.4 1984.74   518.4 1987.26
   534.4 2002.65   558.4 2027.18   573.9    2040   602.4 2055.83     625 2058.33
#Mann= 3 ,-1,0
       0      .1       0   398.4    .045       0   430.4      .1       0
#XS Ineff= 2 , 0
          352.96 1997.55
Permanent Ineff=
       F       F
Bank Sta=398.4,430.4
XS Rating Curve= 0 ,0
Exp/Cntr(USF)=0,0
Exp/Cntr=0.3,0.1

Type RM Length L Ch R = 1 ,17661   ,75.4,87.3,74.9
XS GIS Cut Line= 6
2203331.23026911645047.020338464 2203277.6667951645340.209880366
2203122.61463352645409.278570526 2202957.6955162645537.548995109
2202847.74943799645641.8568129012202921.04682346645754.622021325
#Sta/Elev= 30
       0 2010.77    30.7 2010.25    42.9  2008.3    63.2 2000.47    83.5 1985.83
    95.7 1982.83   132.3 1987.33   217.8 1987.03     238  1988.5   254.3 1983.99
   266.5 1984.88   282.8 1983.16   299.7 1984.16   349.6 1982.54   387.3 1984.62
   452.9 1982.18   506.7 1983.34   532.2 1977.31  563.861975.484     612  1974.4
  638.441975.436   657.6 1981.24   693.6 1982.87   705.8 1981.47   736.9 1981.63
   833.9 1984.43   846.5 1989.38   888.8 2011.63   946.5 2033.12   962.8  2040.9
#Mann= 4 ,-1,0
       0      .1       0  563.86    .045       0  638.44      .1       0
  938.26     .08       0
Bank Sta=563.86,638.44
XS Rating Curve= 0 ,0
Exp/Cntr(USF)=0,0
Exp/Cntr=0.3,0.1

Type RM Length L Ch R = 1 ,17574   ,238.8,195.1,171.2
XS GIS Cut Line= 6
2203255.81853597 645027.286426992203202.25506197645320.475968892
2203047.20290039645389.5446590522202882.28378307645517.815083634
2202772.33770485645622.1229014272202845.63509033645734.888109851
#Sta/Elev= 30
       0 2012.12    42.6  2011.5    75.1 2008.64    83.2  2006.9    91.4 2003.34
   119.8 1983.91     132 1980.94   176.8 1986.65   262.2 1986.81   294.7 1982.92
   372.9 1981.48   422.9 1978.88   486.8 1979.43   525.8 1977.82   543.8 1978.82
   549.5 1978.14     558 1974.84   562.8 1974.26  633.111974.825   733.9 1979.87
   828.3  1982.3   841.9 1981.28   855.8 1982.24     872 1981.68   898.7 1989.92
   905.5 1994.52   922.9 2002.59   932.1 2004.58   951.2 2013.33   962.8 2017.44
#Mann= 3 ,-1,0
       0      .1       0     558    .045       0  633.11      .1       0
Bank Sta=558,633.11
XS Rating Curve= 0 ,0
Exp/Cntr(USF)=0,0
Exp/Cntr=0.3,0.1

Type RM Length L Ch R = 1 ,17378   ,265.8,251.9,246.4
XS GIS Cut Line= 3
2202720.10690718  645223.14610882202760.29756873645623.756251325
2202836.78947296645741.735290063
#Sta/Elev= 30
       0 2029.99    14.1 2031.02    22.1 2030.52    45.8 2019.19    58.3 2014.72
   106.6 2004.23   126.7 1997.63   134.7 1993.36   150.8 1980.87   154.8  1978.8
     170 1974.92   178.9 1975.62   194.3 1973.01   231.2 1972.21   261.4 1973.11
   283.4 1974.92   295.5 1979.06   311.6 1979.03   335.7 1981.41     349 1981.29
   363.9 1982.63   404.3 1982.47   423.8 1981.16     452 1981.84     473 1988.27
   485.4 1995.74   494.9 1996.91   504.4 2002.36   518.7 2008.59   543.2  2017.2
#Mann= 3 ,-1,0
       0      .1       0   194.3    .045       0   261.4      .1       0
Bank Sta=194.3,261.4
XS Rating Curve= 0 ,0
Exp/Cntr(USF)=0,0
Exp/Cntr=0.3,0.1

Type RM Length L Ch R = 1 ,17127   ,179.5,168.6,162.3
XS GIS Cut Line= 2
2202447.36333993645403.4392198842202603.36862273645773.220077079
#Sta/Elev= 30
       0 2031.56    23.3 2029.96    27.9 2028.14    32.3 2024.77    49.6 2009.44
      67  1995.8    75.7 1987.71      80 1984.64    88.7 1981.05    96.6  1974.8
   101.7 1972.59104.69991970.466   106.1 1969.54   110.4 1968.55   125.6 1968.42
   158.2 1969.17   162.5 1969.43166.48991970.432   175.5 1974.23   184.2 1976.21
   205.9 1975.66   236.3 1978.53   297.1  1979.7   323.2 1978.76   349.2 1981.11
   362.2 1980.28   377.5 1980.62   383.9 1979.96   392.6 1977.67   401.3 1978.19
#Mann= 3 ,-1,0
       0      .1       0104.6999    .045       0166.4899      .1       0
Bank Sta=104.6999,166.4899
XS Rating Curve= 0 ,0
Exp/Cntr(USF)=0,0
Exp/Cntr=0.3,0.1

Type RM Length L Ch R = 1 ,16958   ,235.2,219.4,210.7
XS GIS Cut Line= 2
2202275.41668425645521.3348880262202523.26732153645827.058656571
#Sta/Elev= 30
       0 2031.46    20.3  2024.4      26 2023.08    35.8 2016.54    43.1 2015.64
      52 2015.39    56.4 2014.06    58.4  2012.7    71.5 2001.06    83.8 1992.62
    97.1 1982.46   102.8 1976.94   107.9 1972.58   113.1 1969.68   115.5 1968.91
   118.2  1968.5   138.8 1968.29   166.3  1968.4   173.9 1969.01   185.2 1972.46
   205.8 1976.33   216.6 1976.34   236.5 1977.34   276.3 1976.71   299.7 1976.89
   337.8 1978.65   361.6 1979.16   374.6 1978.48     386 1976.61   393.6 1977.18
#Mann= 3 ,-1,0
       0      .1       0   115.5    .045       0   173.9      .1       0
Bank Sta=115.5,173.9
XS Rating Curve= 0 ,0
Exp/Cntr(USF)=0,0
Exp/Cntr=0.3,0.1

Type RM Length L Ch R = 1 ,16739   ,390.8,381.4,371.6
XS GIS Cut Line= 2
2202096.96363021645736.2628708792202409.02448212645901.907413425
#Sta/Elev= 30
       0 2008.36    30.8  2007.4    39.9 2003.24    50.4  1999.4    56.3 1996.32
    65.2 1989.05    71.6  1982.7    78.7  1974.8    80.6 1973.08    82.9  1971.8
    89.7 1969.38    98.7 1969.89109.20971967.522   112.3 1966.73   121.4 1966.41
   130.4 1967.27   156.9 1966.19   165.8 1966.29173.88371967.605   184.8 1970.73
   189.4 1971.58   201.3 1973.08   216.1 1973.06   225.5 1975.51   230.8 1976.24
   261.8 1976.18   311.6 1973.73   325.5 1974.32   343.3 1974.31   353.3 1975.45
#Mann= 3 ,-1,0
       0      .1       0109.2097    .045       0173.8837      .1       0
Bank Sta=109.2097,173.8837
XS Rating Curve= 0 ,0
Exp/Cntr(USF)=0,0
Exp/Cntr=0.3,0.1

Type RM Length L Ch R = 1 ,16357   ,251.4,271.5,291.1
XS GIS Cut Line= 3
2201883.91517576645857.213453151 2202002.4769456 646138.24875943
2202236.17993691646190.649427458
#Sta/Elev= 30
       0 2008.41      13 2002.51    30.7 1995.85    43.4 1993.56    69.4 1985.84
    73.8 1984.27    82.4 1979.65     104  1979.2   112.8 1974.42   117.2 1973.41
   146.7 1970.97   199.7  1971.6   208.3 1972.71   226.1 1973.02   256.1 1971.71
   278.5 1972.16   299.4 1971.62   342.4 1968.23351.44671964.457   356.2  1963.5
   379.2 1963.29   421.5 1963.57429.4738 1964.36   450.2 1971.09   470.7 1972.55
   483.1 1972.49   495.3 1981.25   499.4 1983.25   536.3 1990.96   544.5 1993.76
#Mann= 3 ,-1,0
       0      .1       0351.4467    .045       0429.4738      .1       0
Bank Sta=351.4467,429.4738
XS Rating Curve= 0 ,0
Exp/Cntr(USF)=0,0
Exp/Cntr=0.3,0.1

Type RM Length L Ch R = 1 ,16086   ,469.7,490.6,509.1
XS GIS Cut Line= 2
2201694.59680123645941.3921248492202064.09159288646514.433170145
#Sta/Elev= 30
       0 1999.81    10.3 1991.89      27 1990.12    37.8 1986.14    71.1 1983.08
    99.7 1970.09   104.5 1969.27   142.8 1968.46   168.8 1970.86   180.6 1967.79
   218.7 1968.91   237.7 1968.06   418.6 1970.95   437.6 1970.48   460.6  1966.8
   475.7 1967.38   504.8 1964.73     527 1960.96   539.2 1959.31   561.4 1959.08
   573.9    1961   585.5 1969.78   608.2 1971.39   611.5 1973.26   615.6 1978.85
   630.3 2008.57   634.7 2014.48   645.1    2024   659.8 2035.13   681.8 2046.98
#Mann= 3 ,-1,0
       0      .1       0     527    .045       0   573.9      .1       0
Bank Sta=527,573.9
XS Rating Curve= 0 ,0
Exp/Cntr(USF)=0,0
Exp/Cntr=0.3,0.1

Type RM Length L Ch R = 1 ,15595   ,245.8,241.5,237.9
XS GIS Cut Line= 2
2201642.57707363645962.4893692612201474.35736971646548.357993275
#Sta/Elev= 30
       0 1995.26       7 1993.74    23.6 1987.07    36.1 1983.91    69.4 1980.79
    81.9 1977.88    94.4 1976.42   106.8 1972.34     127 1969.38   223.4 1964.73
   314.9 1963.11   335.7 1964.06   356.5 1963.06   372.7 1963.54   385.5  1958.4
   398.2 1956.01   423.1 1957.37   439.8 1959.68  461.691955.874   473.1 1955.15
  507.091955.887   514.7 1958.96     523 1963.93   540.8 1966.34   544.1 1968.59
   552.1 1979.97   556.3  1984.7   560.5 1987.63   576.4 1990.71   609.5 1994.58
#Mann= 3 ,-1,0
       0      .1       0  461.69    .045       0  507.09      .1       0
Bank Sta=461.69,507.09
XS Rating Curve= 0 ,0
Exp/Cntr(USF)=0,0
Exp/Cntr=0.3,0.1

Type RM Length L Ch R = 1 ,15354   ,292.2,299.1,303.8
XS GIS Cut Line= 2
2201322.50906368645955.6533273342201247.31363239646580.553290756
#Sta/Elev= 30
       0 2015.76    33.8 2002.75      43 1995.63    49.9 1992.08    78.1 1989.66
    90.2 1982.54    98.2 1980.08   130.5 1977.06   158.7 1972.32   170.7 1972.16
   215.1 1966.97   239.2 1961.84   291.6 1959.41   311.8  1960.7   360.1 1958.65
   392.3 1955.78   406.7 1952.08   415.9 1951.16  465.53  1952.1   468.9 1953.56
   476.9  1960.1     481 1961.59   505.1  1961.7   513.2 1964.18   524.9 1970.01
   537.4  1970.6   557.5 1977.76   582.4 1980.66     618 1982.36   629.4 1984.43
#Mann= 3 ,-1,0
       0      .1       0   406.7    .045       0  465.53      .1       0
Bank Sta=406.7,465.53
XS Rating Curve= 0 ,0
Exp/Cntr(USF)=0,0
Exp/Cntr=0.3,0.1

Type RM Length L Ch R = 1 ,15054   ,557.8,549.3,539.8
XS GIS Cut Line= 2
2201097.31320574645945.0873309242200886.55518588646625.700385884
#Sta/Elev= 30
       0 2019.73    20.2 2022.62    25.2 2021.75    37.8  2013.8    92.2 1996.22
   142.5 1982.41     176 1974.43   188.5 1973.01   205.3 1961.27   213.7 1958.36
   226.2 1957.37     243 1958.09   293.2 1957.23   314.2 1954.42   330.9 1956.54
  358.841949.819   385.3 1948.79   431.4 1949.92   439.8 1950.85   452.3 1955.92
   460.7 1957.12   531.9 1958.59   561.2 1955.92     578 1957.75   590.5 1956.53
     645 1958.49   665.9 1957.47   674.3 1961.01   703.6 1981.36   712.5 1986.35
#Mann= 4 ,-1,0
       0      .1       0  358.84    .045       0   431.4      .1       0
     600     .08       0
#XS Ineff= 2 , 0
          328.56 1972.82
Permanent Ineff=
       F       F
Bank Sta=358.84,431.4
XS Rating Curve= 0 ,0
Exp/Cntr(USF)=0,0
Exp/Cntr=0.3,0.1

Type RM Length L Ch R = 1 ,14505   ,524.3,524.5,521.5
XS GIS Cut Line= 2
2200453.43778727 646035.96464224 2200418.6337106646614.099026992
#Sta/Elev= 30
       0 1996.85    21.3 1990.78    68.2 1979.91    81.4 1974.58   101.4 1972.58
   113.4 1967.01   129.4 1963.37   137.5 1960.62   144.9 1957.05   157.5 1949.48
  172.481945.848   201.6  1944.8   241.7 1944.99  253.53 1945.78   265.7  1949.8
   277.7 1951.02   285.8 1953.95   293.7 1954.36   341.8 1952.91   389.9 1953.26
     430 1952.55     454 1951.47   477.5 1947.12   498.1 1947.32   510.1 1952.92
   526.2 1954.02   530.2 1954.96   542.2 1963.24   570.2 1976.02   579.2  1981.6
#Mann= 4 ,-1,0
       0      .1       0  172.48    .045       0  253.53      .1       0
     490     .08       0
#XS Ineff= 2 , 0
                           403.3         1957.23
Permanent Ineff=
       F       F
Bank Sta=172.48,253.53
XS Rating Curve= 0 ,0
Exp/Cntr(USF)=0,0
Exp/Cntr=0.3,0.1

Type RM Length L Ch R = 1 ,13981   ,513.8,514.4,506.1
XS GIS Cut Line= 2
 2199923.6423979  646043.69888152199917.84171845646596.696988655
#Sta/Elev= 30
       0 1996.26    29.5 1985.77    41.5  1977.9    65.5 1975.64    69.5  1974.2
    77.5 1968.52    89.5  1963.1   113.5 1955.49   137.5 1951.08   149.5 1944.49
  156.49 1942.44   165.5 1941.32   193.5 1941.93   205.5 1941.04   216.3 1942.43
   237.5 1946.31   273.5  1946.2   301.5 1947.53   313.5 1947.22   341.5 1943.91
   361.5 1948.72   381.5 1948.54   397.5 1946.08   453.5 1942.25   457.5 1943.17
   473.5  1952.5   489.5 1954.17   505.5  1963.1   521.5 1970.22     553 1981.13
#Mann= 4 ,-1,0
       0      .1       0  156.49    .045       0   216.3      .1       0
     480     .08       0
#XS Ineff= 2 , 0
                          376.24            1955
Permanent Ineff=
       F       F
Bank Sta=156.49,216.3
XS Rating Curve= 0 ,0
Exp/Cntr(USF)=0,0
Exp/Cntr=0.3,0.1

Type RM Length L Ch R = 1 ,13466   ,184.3,186.2,185.4
XS GIS Cut Line= 2
2199399.64768797646161.6460302292199488.59143947646617.966146623
#Sta/Elev= 30
       0 1979.04     3.6 1976.72    15.8 1975.36    19.9 1973.87    36.2 1962.25
    56.6 1951.47   75.871938.125      81 1936.72     105 1936.62   121.8 1938.15
   129.9 1940.93   142.2  1942.7   191.1 1942.44   219.6 1938.34   252.4 1941.71
   292.3 1939.36   297.4 1940.59   309.2 1947.77   313.3 1948.55   329.6 1948.51
   337.9 1949.82     350 1950.09   358.1 1953.28   366.3 1954.79   386.7 1955.17
   407.1 1957.75   435.6 1963.57   443.7 1964.06   453.6 1967.15   464.9  1969.2
#Mann= 4 ,-1,0
       0      .1       0   75.87    .045       0   121.8      .1       0
  464.91     .08       0
Bank Sta=75.87,121.8
XS Rating Curve= 0 ,0
Exp/Cntr(USF)=0,0
Exp/Cntr=0.3,0.1

Type RM Length L Ch R = 1 ,13280   ,279.8,275.1,261.4
XS GIS Cut Line= 2
2199219.53677967646201.4554759242199317.20008723646671.919581166
#Sta/Elev= 30
       0 1968.28    10.5  1962.6    28.3 1950.68    40.6 1944.15    52.8 1941.46
      68  1941.2    82.31939.185   114.1 1936.47   126.4  1936.9   140.91939.312
   163.1 1940.26   175.4 1941.82   199.9 1939.78   240.7 1938.57   261.2 1936.45
   265.3 1936.75   273.4  1939.6   281.6 1944.55   285.7 1946.04   297.9 1944.75
   310.2 1946.56   321.7 1946.26   334.7 1949.06   363.3 1952.67   404.2  1955.3
   428.7 1955.43   440.9 1956.59   449.1 1958.52   465.4 1957.94   480.5 1960.42
#Mann= 3 ,-1,0
       0      .1       0    82.3    .045       0   140.9      .1       0
Bank Sta=82.3,140.9
XS Rating Curve= 0 ,0
Exp/Cntr(USF)=0,0
Exp/Cntr=0.3,0.1

Type RM Length L Ch R = 1 ,13005   ,323.6,327.7,316.4
XS GIS Cut Line= 2
2198957.00100666646333.7735055232199185.93220072646737.028452873
#Sta/Elev= 30
       0 1965.81     3.9 1966.49     8.5 1965.31    13.6 1962.31    22.6 1954.98
    37.1 1947.65    49.9 1937.76    63.5 1934.07    72.9 1933.13    82.1 1935.46
    95.9 1936.88   103.7 1936.79   111.2 1935.64   144.2 1934.55   152.3 1935.53
   160.3 1936.91   178.7 1933.64   200.9 1934.29   224.9  1942.1   252.3 1941.41
     263 1942.67   275.3 1942.05   321.3 1945.79   336.4 1948.57   362.7 1951.84
   376.5 1955.12   390.3 1956.87   404.1 1956.23   417.9 1956.98   463.7 1965.03
#Mann= 4 ,-1,0
       0      .1       0   111.2    .045       0   152.3      .1       0
     440     .08       0
Bank Sta=111.2,152.3
XS Rating Curve= 0 ,0
Exp/Cntr(USF)=0,0
Exp/Cntr=0.3,0.1

Type RM Length L Ch R = 1 ,12677   ,237.5,242.8,244.9
XS GIS Cut Line= 2
2198671.36208562646516.4984035412199003.20730271646858.845051552
#Sta/Elev= 30
       0 1944.77    37.8 1941.34    58.6 1941.55    73.4 1940.24    78.9 1939.02
    94.4 1933.73   101.2 1932.02   129.1 1929.67   156.3 1928.37   173.6 1929.15
   187.8 1928.63   201.5 1929.71   218.2 1929.66   227.4 1930.42   235.8 1932.08
   244.3 1935.56   252.8  1936.2   259.8 1937.41   275.4 1936.89   279.5 1937.89
   303.7 1946.64   323.5 1952.79     332 1955.13   346.3 1958.02   363.2 1960.46
   385.3 1964.43     415 1966.56   452.2 1972.38   467.8  1974.3   476.8 1974.81
#Mann= 3 ,-1,0
       0      .1       0   129.1    .045       0   201.5      .1       0
Bank Sta=129.1,201.5
XS Rating Curve= 0 ,0
Exp/Cntr(USF)=0,0
Exp/Cntr=0.3,0.1

Type RM Length L Ch R = 1 ,12434   ,253.3,248.7,244.9
XS GIS Cut Line= 2
2198458.00405796646606.3647877322198719.03463301 646935.06995632
#Sta/Elev= 30
       0 1957.41    17.8 1954.37    29.1 1953.41    71.9 1943.93    83.3 1943.39
     100 1940.51   117.4 1939.49     126 1940.03   136.4 1937.33   148.7 1935.54
   168.7 1934.25   174.4 1932.86   183.6 1929.26   194.71926.591   260.8 1925.88
  271.471926.578   276.9 1926.96   292.9  1926.4   299.4 1926.84   318.7  1931.2
   333.8 1933.22   345.2 1936.12   359.4 1936.45   363.7 1938.15   370.8 1945.29
   376.1  1948.9     385 1951.82   389.4 1952.72     402 1953.75   419.7 1953.46
#Mann= 3 ,-1,0
       0      .1       0   194.7    .045       0  271.47      .1       0
Bank Sta=194.7,271.47
XS Rating Curve= 0 ,0
Exp/Cntr(USF)=0,0
Exp/Cntr=0.3,0.1

Type RM Length L Ch R = 1 ,12186   ,346,339.7,335.1
XS GIS Cut Line= 2
2198272.61700144646811.1764026592198587.65992906647118.868328634
#Sta/Elev= 30
       0 1952.89     8.6 1952.63    31.5 1950.49    48.7 1947.91    60.1 1947.89
    77.3 1946.36    88.7 1944.01   128.8  1939.9   140.3 1937.03     151 1929.92
   153.8 1928.83   167.1 1926.42   176.5 1924.01   218.9 1923.45   234.2 1924.06
   264.2 1927.09     267 1926.86   275.5 1924.46   278.9 1924.17   289.1 1925.99
   300.9 1930.52   312.5 1930.93   329.2 1929.22   334.9 1929.16   357.2 1931.49
   371.7 1934.26     383  1935.4   399.9 1935.86   424.3 1933.15   440.4 1934.67
#Mann= 3 ,-1,0
       0      .1       0   176.5    .045       0   234.2      .1       0
#XS Ineff= 2 , 0
                          310.99         1936.47
Permanent Ineff=
       F       F
Bank Sta=176.5,234.2
XS Rating Curve= 0 ,0
Exp/Cntr(USF)=0,0
Exp/Cntr=0.3,0.1

Type RM Length L Ch R = 1 ,11846   ,349.8,350.9,347.9
XS GIS Cut Line= 3
2198018.39313189647061.0213092892198471.96943128647403.882134025
2198857.14955143647304.880324699
#Sta/Elev= 30
       0 1956.82    22.3    1954    52.8 1951.68    72.8 1948.51    82.5  1944.3
   107.5 1926.93   129.9 1921.39   152.7    1921   201.3 1921.39   217.8 1924.09
     288 1926.88   335.5 1927.44   358.3 1925.75   386.9 1926.29   404.9 1928.04
   421.2 1928.36     444 1930.87   517.7 1931.27   558.8 1928.07   577.1 1929.75
   593.6 1928.45   642.9 1930.76   655.5 1929.52   684.4 1929.19   717.5  1930.2
   807.5 1929.88   903.3 1936.45   919.8 1936.53   948.8 1939.56   966.3 1942.49
#Mann= 3 ,-1,0
       0      .1       0   129.9    .045       0   201.3      .1       0
Bank Sta=129.9,201.3
XS Rating Curve= 0 ,0
Exp/Cntr(USF)=0,0
Exp/Cntr=0.3,0.1

Type RM Length L Ch R = 1 ,11495   ,466.5,458,434.8
XS GIS Cut Line= 3
2197819.35007464647348.2563502942198265.78636847647660.517801714
2198580.48736248647648.320088768
#Sta/Elev= 30
       0  1960.4    20.5    1957    25.4 1954.99      30 1952.11    59.6 1925.95
    64.4  1922.4    70.2 1919.93      84 1918.94   137.7 1919.89   147.4 1921.19
   179.3 1922.11   196.6 1924.88   228.2 1922.56   280.8 1924.43   336.6 1921.37
   351.7 1923.99   368.9 1925.15   434.3 1924.33   449.3 1926.85   489.1 1927.88
   532.6 1926.42   544.1 1927.17   571.2 1926.73   589.6 1925.06   606.3 1926.83
   619.2 1925.72   639.3  1927.8   675.3  1926.2   759.4 1925.58   859.7 1927.06
#Mann= 3 ,-1,0
       0      .1       0    70.2    .045       0   137.7      .1       0
#XS Ineff= 2 , 0
                          485.63         1933.97
Permanent Ineff=
       F       F
Bank Sta=70.2,137.7
XS Rating Curve= 0 ,0
Exp/Cntr(USF)=0,0
Exp/Cntr=0.3,0.1

Type RM Length L Ch R = 1 ,11037   ,292.6,299.7,302.7
XS GIS Cut Line= 3
2197736.03481613647646.2220821412198137.95921588647925.435050105
2198682.15773943647811.615751063
#Sta/Elev= 30
       0 1943.49    19.7 1939.71    34.3 1930.15      44 1920.58    48.9  1918.9
    82.3 1920.76   126.8 1919.25   180.5 1921.59   214.5 1920.32     234 1917.34
     268 1915.84   277.8 1915.43     304 1915.83   321.2 1920.19   327.7 1919.93
   341.1 1922.15   414.2 1922.97   467.7 1925.94   499.8 1922.65   517.8 1923.81
   536.6 1923.04   548.9 1924.53   622.4 1923.78   634.7 1924.66   708.2 1923.45
   732.8 1921.42   847.2 1923.56     870 1925.53   903.8 1924.75  1045.4 1926.58
#Mann= 5 ,-1,0
       0      .1       0     268    .045       0     304      .1       0
  619.39     .07       0  649.39      .1       0
#XS Ineff= 2 , 0
                           463.1         1930.82
Permanent Ineff=
       F       F
Bank Sta=268,304
XS Rating Curve= 0 ,0
Exp/Cntr(USF)=0,0
Exp/Cntr=0.3,0.1

Type RM Length L Ch R = 1 ,10738   ,389.2,392.8,389.3
XS GIS Cut Line= 3
2197547.52160209647815.1726041582197969.00869386648147.738368548
2198155.74348135648610.129270909
#Sta/Elev= 30
       0 1952.99    50.3  1938.5    67.4  1937.9    95.9 1919.61   127.2 1916.13
   158.5 1919.86   192.7 1918.66     225 1920.96   266.8 1917.57   296.4 1919.45
   335.1 1918.89   343.7 1917.28   369.3 1919.87   408.4 1918.81   417.7 1917.73
   423.7 1915.13   477.5 1915.15   494.6 1921.47   555.8 1921.44   583.5 1918.95
   706.7 1918.02   758.5 1915.22   814.5 1915.97   836.1 1913.41   857.7 1914.52
   870.6 1919.22   887.2 1922.04   909.4 1930.44     943 1934.15  1035.6 1952.84
#Mann= 3 ,-1,0
       0      .1       0   423.7    .045       0   477.5      .1       0
#XS Ineff= 2 , 0
                          558.42         1926.43
Permanent Ineff=
       F       F
Bank Sta=423.7,477.5
XS Rating Curve= 0 ,0
Exp/Cntr(USF)=0,0
Exp/Cntr=0.3,0.1

Type RM Length L Ch R = 1 ,10345   ,344.4,366.8,393.5
XS GIS Cut Line= 3
2197438.78143072 647862.999836622197587.59352866 648331.39201375
2197909.61315044648602.181241153
#Sta/Elev= 30
       0 1956.25    18.8 1949.49    31.5 1940.97    41.1 1937.09    65.2 1922.25
    77.8 1917.64   195.3  1918.1   248.1 1915.03   275.1 1916.78   305.4 1915.13
   333.9 1910.06   367.4 1914.53   430.4 1914.73   472.4 1917.28   506.7 1916.82
   518.7 1916.41   531.5 1910.85   544.5 1909.82     602 1910.76   624.8  1914.8
   659.5 1914.02   699.3 1917.45   737.9  1914.9   757.2 1915.75   786.3 1911.36
   816.8 1913.03   836.1 1917.23   862.2 1931.09   882.1 1935.56   912.2 1937.73
#Mann= 3 ,-1,0
       0      .1       0   531.5    .045       0     602      .1       0
#XS Ineff= 2 , 0
          272.68 1922.21  700.12         1919.61
Permanent Ineff=
       F       F
Bank Sta=531.5,602
XS Rating Curve= 0 ,0
Exp/Cntr(USF)=0,0
Exp/Cntr=0.3,0.1

Type RM Length L Ch R = 1 ,9978    ,227.1,244.5,265.4
XS GIS Cut Line= 2
2197408.25104729 647877.127927672197393.92838199648786.617174092
#Sta/Elev= 30
       0 1954.76    20.1 1947.21    64.1 1921.42    76.1 1916.85    84.1 1915.81
   176.1 1917.52   244.1 1914.76   292.1 1915.91   336.1 1915.03   360.1 1913.19
   376.1 1914.75   460.1 1914.12   476.1 1913.46   496.1 1908.53   512.1 1908.19
   548.1 1912.67   572.1 1910.31   636.1 1913.21   676.1 1913.49   700.1 1911.47
   724.1 1911.34  731.341907.515   752.4 1906.22   788.5 1907.57   800.2 1914.45
   820.2 1917.48   836.2 1928.57   852.2 1936.41   890.1  1941.6   909.6  1942.4
#Mann= 3 ,-1,0
       0      .1       0  731.34    .045       0   788.5      .1       0
#XS Ineff= 2 , 0
          443.38 1919.26
Permanent Ineff=
       F       F
Bank Sta=731.34,788.5
XS Rating Curve= 0 ,0
Exp/Cntr(USF)=0,0
Exp/Cntr=0.3,0.1

Type RM Length L Ch R = 1 ,9733    ,367.1,367.6,365.3
XS GIS Cut Line= 3
2197359.00838805647875.639106774 2197323.4398571 648348.70056842
2197083.35227319648638.584095669
#Sta/Elev= 30
       0 1957.05    33.6 1948.57    61.7 1933.01    77.8 1922.16    93.8 1915.76
   101.8 1914.28   218.2 1917.04   334.5 1913.74   358.5 1911.72   395.8 1913.71
   430.8 1913.24     514 1914.44   552.9 1913.22   573.6 1914.09   582.2 1913.53
   599.2  1908.6   620.4 1906.56   627.6 1904.95   655.1  1904.5   690.1  1904.9
     693 1905.45   703.5 1911.34   719.1 1912.71   724.1 1916.61   729.9 1922.64
   734.7 1925.02   765.9  1929.6   817.8 1933.44   833.4 1933.55   850.8 1935.96
#Mann= 4 ,-1,0
       0      .1       0   627.6    .045       0   690.1      .1       0
   704.4     .08       0
Bank Sta=627.6,690.1
XS Rating Curve= 0 ,0
Exp/Cntr(USF)=0,0
Exp/Cntr=0.3,0.1

Type RM Length L Ch R = 1 ,9366    ,457.2,459,460.1
XS GIS Cut Line= 2
2197237.97047097647872.0884713612196816.24754831 648391.94817477
#Sta/Elev= 30
       0 1946.58    47.6 1936.77    67.5 1927.34    84.5 1916.69    90.2 1914.07
   119.9 1908.99   135.3 1908.27   161.1 1910.23   243.5 1910.36   260.8 1911.07
   301.3 1909.81   345.7 1910.72     362 1910.03   371.1 1906.82   377.5 1905.87
     398 1906.44   421.9 1904.85   431.5 1902.11   454.7 1900.84   502.6 1901.26
  510.461902.074   525.3 1907.12   531.9 1906.92   542.4  1908.5   559.4 1907.19
   574.3  1909.1   596.4 1914.35   634.9 1919.02   645.2 1919.11   669.4 1922.54
#Mann= 4 ,-1,0
       0      .1       0   431.5    .045       0  510.46      .1       0
     540     .08       0
#XS Ineff= 2 , 0
                          542.25         1910.64
Permanent Ineff=
       F       F
Bank Sta=431.5,510.46
XS Rating Curve= 0 ,0
Exp/Cntr(USF)=0,0
Exp/Cntr=0.3,0.1

Type RM Length L Ch R = 1 ,8907    ,950,946.8,947.8
XS GIS Cut Line= 2
2196871.23732713647623.5284131482196456.46726058648096.511822369
#Sta/Elev= 30
       0 1920.39      60 1910.89    95.6 1903.19   122.4 1901.99   138.1 1902.15
   151.2 1903.98   170.6 1903.66   181.9 1902.36     217 1902.67   255.6 1905.44
   271.6 1901.22   278.3 1900.65   295.3 1902.32   342.7 1901.81   350.5 1901.16
  358.09 1898.93   390.6 1898.33     437 1898.94   456.9 1904.53   470.4 1902.73
   482.4 1903.56   493.7 1902.82   507.9 1904.12   519.2 1902.32   527.7 1902.27
   534.2 1904.09   550.4 1913.68   556.7 1915.66   612.8 1919.82   629.1 1922.25
#Mann= 4 ,-1,0
       0      .1       0  358.09    .045       0     437      .1       0
  629.08     .08       0
#XS Ineff= 2 , 0
          254.76 1909.31
Permanent Ineff=
       F       F
Bank Sta=358.09,437
XS Rating Curve= 0 ,0
Exp/Cntr(USF)=0,0
Exp/Cntr=0.3,0.1

Type RM Length L Ch R = 1 ,7960    ,573.1,567.7,553.5
XS GIS Cut Line= 2
2196336.10818039646870.1060028072195962.85816424647753.220420105
#Sta/Elev= 30
       0 1913.39    10.1 1910.73    26.7 1903.27    38.1 1902.11    72.8 1901.36
    98.9 1908.57   173.2 1906.37   181.4  1903.3   190.1 1894.64   194.4 1892.64
     216 1892.12   246.5 1892.69   263.9 1895.14   289.9 1896.37   333.4 1896.57
   396.1 1893.65   460.2 1896.55     481 1898.83   534.1 1899.05   715.5    1899
     799 1895.37   815.4 1896.95   837.1 1893.56   858.8 1893.07   867.5 1894.53
   871.9 1896.84   883.4 1906.02   893.6 1910.76   933.3 1936.64   958.8 1949.93
#Mann= 4 ,-1,0
       0      .1       0   194.4    .045       0   246.5      .1       0
     900     .08       0
Bank Sta=194.4,246.5
XS Rating Curve= 0 ,0
Exp/Cntr(USF)=0,0
Exp/Cntr=0.3,0.1

Type RM Length L Ch R = 1 ,7392    ,622.8,620.5,610.1
XS GIS Cut Line= 2
2195735.98070345646701.7775641512195711.58527755647616.606035108
#Sta/Elev= 30
       0 1911.19    31.4 1906.78    95.4 1904.58     120 1892.89   131.4 1888.74
   151.5    1888   183.5 1888.79   199.5 1892.84   251.5 1893.81   335.5 1892.88
   357.8 1889.74   371.5 1890.99   391.5 1894.97   443.5 1894.41   475.6 1890.59
   494.2    1892   535.6 1891.09   575.6 1894.63   599.6 1893.58   651.6 1895.53
     693 1893.39     732 1893.86   755.7 1891.62   774.8 1893.46   811.7  1890.8
   819.7 1894.64   835.7 1907.97   855.7 1928.03   883.7 1958.18   915.2 1980.04
#Mann= 4 ,-1,0
       0      .1       0   131.4    .045       0   183.5      .1       0
     800     .08       0
Bank Sta=131.4,183.5
XS Rating Curve= 0 ,0
Exp/Cntr(USF)=0,0
Exp/Cntr=0.3,0.1

Type RM Length L Ch R = 1 ,6772    ,758.3,746.5,741.6
XS GIS Cut Line= 2
 2195103.9772658646840.8509192592195289.64144559647648.342748816
#Sta/Elev= 30
       0  1910.8      25 1907.05    93.9 1900.13    98.8 1898.15   113.9 1885.82
  118.031883.782   160.4 1882.69     184 1883.78   193.2 1886.68   217.9 1890.18
   275.3  1887.8   380.9 1888.55   406.7 1886.84     419 1884.83   435.4 1885.98
   451.8 1885.04   488.8 1887.67   529.8 1886.84   599.6  1890.5     616 1887.95
   648.8 1889.62   667.9 1888.36   707.9 1889.66   718.6 1888.66   727.9  1886.1
   747.3    1887   767.9 1891.23   792.5 1912.43   804.8 1924.51   828.6  1944.1
#Mann= 3 ,-1,0
       0      .1       0  118.03    .045       0     184      .1       0
Bank Sta=118.03,184
XS Rating Curve= 0 ,0
Exp/Cntr(USF)=0,0
Exp/Cntr=0.3,0.1

Type RM Length L Ch R = 1 ,6025    ,690.6,677.5,668.2
XS GIS Cut Line= 2
2194357.88114825647110.3409150572194721.71453995647805.262693221
#Sta/Elev= 30
       0  1918.1    42.3 1909.56    70.9 1905.54   111.6 1902.05   125.1 1899.26
   143.2 1898.83   165.7 1895.84   175.7 1893.18   194.7 1893.03   201.9 1889.52
   211.9  1881.4   220.5 1878.14   260.6 1876.95   280.9 1877.05   289.5 1878.15
   300.2 1880.42   337.3 1880.17   353.5 1883.06   364.4 1883.77   581.1 1879.31
   599.2 1880.78   612.7 1879.76   621.8 1883.01   626.3  1883.4   639.8 1879.95
   657.9 1879.42   676.5 1882.15     694 1892.61   707.6 1897.98   784.4 1909.86
#Mann= 6 ,-1,0
       0      .1       0     110     .06       0     220      .1       0
   220.5    .045       0   289.5      .1       0     780     .08       0
Bank Sta=220.5,289.5
XS Rating Curve= 0 ,0
Exp/Cntr(USF)=0,0
Exp/Cntr=0.3,0.1

Type RM Length L Ch R = 1 ,5348    ,467.1,462.8,454.3
XS GIS Cut Line= 2
2193728.44938059647612.4309956152194318.17193528648014.450120733
#Sta/Elev= 30
       0 1919.59    28.7  1918.1    69.4 1904.79   138.5 1890.02   147.2 1887.12
   155.8 1881.52   170.2  1875.2   198.2 1873.85   242.8 1876.07   256.2  1875.7
   273.8 1872.93   299.7 1872.93   314.3 1872.56   360.2 1873.49   374.6 1874.58
   386.1 1877.14   420.6 1876.85   446.5 1879.52   464.4 1875.66   488.6 1875.75
   504.1 1878.54   519.7  1875.2   546.7 1875.99   576.1 1873.86   596.2 1876.82
   610.6  1881.9   619.2 1886.67   633.6 1891.11     676 1896.32   713.7  1902.8
#Mann= 5 ,-1,0
       0      .1       0      20     .06       0     130      .1       0
   273.8    .045       0   299.7      .1       0
Bank Sta=273.8,299.7
XS Rating Curve= 0 ,0
Exp/Cntr(USF)=0,0
Exp/Cntr=0.3,0.1

Type RM Length L Ch R = 1 ,4885    ,355.7,355.9,354.3
XS GIS Cut Line= 2
2193499.38013186648048.9911895262194094.48687499648336.876762015
#Sta/Elev= 30
       0 1983.54    21.7 1983.78      32 1980.47    58.6 1959.13      72 1952.66
    94.2 1937.97   129.7 1917.22   135.5 1912.31     152 1893.27   156.4 1889.43
   186.4 1869.43   214.2 1868.19   264.3 1869.36   276.3 1872.18   291.2  1871.2
   309.2  1872.4   356.4 1872.56     383  1875.5   396.4 1873.63   418.6 1873.93
   431.9 1875.81     444 1874.75     463 1876.92   485.9 1883.01   498.5 1888.31
   521.8 1888.31   554.8 1890.86   609.6 1890.99   629.6 1896.67   661.1 1901.56
#Mann= 4 ,-1,0
       0     .06       0     100      .1       0   186.4    .045       0
   264.3      .1       0
Bank Sta=186.4,264.3
XS Rating Curve= 0 ,0
Exp/Cntr(USF)=0,0
Exp/Cntr=0.3,0.1

Type RM Length L Ch R = 1 ,4529    ,327.6,363.5,401.4
XS GIS Cut Line= 3
2193373.74900971 648231.580364622193495.67062269648442.344083196
2193829.30108304648597.345203584
#Sta/Elev= 30
       0 1942.79      25    1931    36.8 1923.58    60.8  1913.7   108.1 1886.28
   131.2 1878.37   145.1 1876.17   212.5 1873.14   257.3 1873.82   264.1 1872.69
   276.1 1867.64   282.1 1866.03   305.8 1865.19   345.5 1865.28     354 1866.05
   360.4 1867.81   367.5 1868.58   390.6 1868.44   402.8 1870.37   420.5 1869.68
   460.2 1874.83   474.9 1874.66   477.9 1875.15   486.6 1879.28   499.9 1880.39
     520 1885.74   535.1 1885.25   561.6  1892.9   574.8 1890.83   611.4 1893.61
#Mann= 3 ,-1,0
       0      .1       0   282.1    .045       0     354      .1       0
Bank Sta=282.1,354
XS Rating Curve= 0 ,0
Exp/Cntr(USF)=0,0
Exp/Cntr=0.3,0.1

Type RM Length L Ch R = 1 ,4166    ,668.2,670.3,650.2
XS GIS Cut Line= 2
2193296.24844951648288.2880915912193300.97409343648947.987982022
#Sta/Elev= 30
       0 1919.21    60.9 1888.13    84.9 1879.32    92.9 1875.39   108.9 1872.33
   280.9 1872.04   288.9 1871.54   300.9 1868.73   320.9 1868.61   368.9  1871.8
   380.9 1870.24   384.9 1866.81   392.9 1863.54   400.9 1862.18   456.9 1863.59
   460.9 1865.29   472.9 1873.66   488.9 1874.56   492.9 1877.61   500.9 1888.46
   504.9 1891.14   512.9 1894.13   516.9 1895.26   532.8 1894.95   540.9 1896.46
   556.9 1903.34   576.9 1906.85   592.9 1912.84   616.4 1917.08   659.7 1928.82
#Mann= 3 ,-1,0
       0      .1       0   392.9    .045       0   456.9      .1       0
Bank Sta=392.9,456.9
XS Rating Curve= 0 ,0
Exp/Cntr(USF)=0,0
Exp/Cntr=0.3,0.1

Type RM Length L Ch R = 1 ,3495    ,324.1,327.7,324
XS GIS Cut Line= 3
2192602.75003027648254.2829344492192738.87969035648527.838727567
2192850.37636432648916.780613516
#Sta/Elev= 30
       0 1970.03    33.1 1957.64    48.1 1947.26    80.8 1943.74   101.5    1931
   137.3 1915.25   155.1 1898.12   164.8 1890.71   190.9 1876.98   209.1 1864.53
   231.1 1859.89   262.4 1858.93   280.2 1860.03   292.6 1862.43   302.6 1868.83
   315.3 1864.37   327.8 1863.11   444.3 1863.05   456.7 1865.49   473.4 1862.25
   506.7 1861.99   535.8 1867.07   556.6 1866.65   581.6 1870.79   610.7  1871.7
   631.1 1877.36     644 1887.19     657 1888.49   673.1 1899.19   710.2 1913.68
#Mann= 4 ,-1,0
       0     .06       0     120      .1       0   231.1    .045       0
   280.2      .1       0
Bank Sta=231.1,280.2
XS Rating Curve= 0 ,0
Exp/Cntr(USF)=0,0
Exp/Cntr=0.3,0.1

Type RM Length L Ch R = 1 ,3168    ,488.1,476.2,469.8
XS GIS Cut Line= 2
2192337.09584292648461.4839501082192659.35581213649045.848694266
#Sta/Elev= 30
       0 1922.13    14.7 1921.09    36.2 1911.41    45.3 1910.17   105.1 1891.65
   109.3 1889.73   122.3  1879.6   128.6 1876.56     155 1871.76   159.5 1868.91
  171.69 1857.19   218.9 1855.66   255.5 1855.96   261.1 1857.23   269.2 1862.28
   278.8 1864.03   378.9 1865.38   397.1 1866.17   412.3 1868.65   434.8 1865.56
   452.5 1866.21   473.1 1870.18   520.4 1870.73   552.6 1878.24   584.3 1880.39
     598 1884.89   611.8 1883.95   623.3 1888.14   643.7 1898.79   667.3 1901.31
#Mann= 7 ,-1,0
       0      .1       0      30     .06       0     140      .1       0
  171.69    .045       0   261.1      .1       0     370     .03       0
     480      .1       0
Bank Sta=171.69,261.1
XS Rating Curve= 0 ,0
Exp/Cntr(USF)=0,0
Exp/Cntr=0.3,0.1

Type RM Length L Ch R = 1 ,2691    ,365.7,362,356.4
XS GIS Cut Line= 2
2191954.68067947648826.7119152072192399.39943697649275.727472299
#Sta/Elev= 30
       0 1890.84     3.5 1890.14    14.1 1884.14    19.2 1882.52    59.4 1874.26
    87.4 1869.86      99 1863.28   115.8 1859.81   130.1 1852.92   135.7 1851.64
   152.7 1851.39     167  1851.4   175.3 1852.95   186.7 1857.01   217.8 1859.65
   246.5 1867.71   256.8 1869.38   277.2 1868.55   325.2 1863.02   348.9 1863.41
   380.7 1862.38   434.1 1863.19   485.3 1865.72   496.7 1865.33   502.3 1866.84
   540.2 1883.99   583.3 1886.41     599 1889.06   617.1 1893.64     632 1894.52
#Mann= 6 ,-1,0
       0     .06       0      80      .1       0   130.1    .045       0
   175.3      .1       0     350     .03       0     630      .1       0
Bank Sta=130.1,175.3
XS Rating Curve= 0 ,0
Exp/Cntr(USF)=0,0
Exp/Cntr=0.3,0.1

Type RM Length L Ch R = 1 ,2329    ,198.9,195.7,189.4
XS GIS Cut Line= 3
2191785.95031987648897.3871147142191757.30498927649159.969311844
2192251.43694205649501.326168113
#Sta/Elev= 30
       0 1894.73    20.3 1889.41    48.1 1887.11    56.1 1885.15    84.3 1885.25
   108.4 1882.59   152.7 1881.32   217.1 1876.02   264.1 1868.58   296.8 1868.04
   306.5 1866.38     316 1862.05     326 1860.78     339 1851.81   345.4 1850.57
   389.2 1850.42  399.581851.712   422.3 1865.84   428.1 1867.75   528.7 1859.23
   577.6 1858.15   651.7 1858.24   729.5 1862.05   758.8 1865.88   768.4 1865.49
     783 1871.02   793.3 1872.21   830.6 1887.19   841.3 1890.05   864.7 1902.66
#Mann= 7 ,-1,0
       0      .1       0      80     .06       0  284.14      .1       0
     339    .045       0  399.58      .1       0  464.14     .03       0
  764.14      .1       0
#XS Ineff= 2 , 0
                          438.94         1873.62
Permanent Ineff=
       F       F
Bank Sta=339,399.58
XS Rating Curve= 0 ,0
Exp/Cntr(USF)=0,0
Exp/Cntr=0.3,0.1

Type RM Length L Ch R = 1 ,2134    ,254.2,232.5,215.2
XS GIS Cut Line= 2
2191470.61630211649254.5158821732192137.00340004649576.041174556
#Sta/Elev= 30
       0 1878.72    50.6 1876.08     120 1869.39   166.1 1863.96   192.7  1859.2
   214.9 1858.01   241.6 1858.72   263.8 1854.41   275.8 1850.07     286 1849.48
   337.5  1850.1   344.7 1854.52   350.7 1856.87   374.6  1859.8   383.6 1858.28
   422.6 1856.67   458.5 1857.06   485.5  1855.9   512.4 1857.22   576.8 1858.41
   605.7 1858.43   619.1 1856.64   632.4 1856.91   636.8 1857.48   659.2 1864.07
   676.8 1865.74   698.2 1866.14   705.7 1867.35   725.2 1871.77   739.9 1876.94
#Mann= 8 ,-1,0
       0      .1       0      10     .06       0     120      .1       0
   275.8    .045       0   337.5      .1       0     450     .07       0
     500    .025       0     550      .1       0
Bank Sta=275.8,337.5
XS Rating Curve= 0 ,0
Exp/Cntr(USF)=0,0
Exp/Cntr=0.3,0.1

Type RM Length L Ch R = 1 ,1901    ,41.6,39.6,52.5
XS GIS Cut Line= 5
 2191205.8823753649635.0043775612191446.98057448649627.843044912
2191692.85299543649580.1008272522191836.07964841649484.616391932
2192127.30717614649582.487938135
#Sta/Elev= 30
       0 1885.42    66.5 1877.33    87.1 1872.15   162.4 1871.15   186.4 1867.55
   206.4 1862.33   230.4 1859.94   368.7 1858.66     385  1856.5     398 1851.03
   405.4 1849.33   417.6 1849.26   450.2 1849.33  463.051851.006   474.7 1856.06
   482.8 1857.86   547.4 1857.37   577.4  1855.2   612.3    1856   662.8 1855.12
   781.2 1858.47   828.3 1858.51   841.2 1856.64   850.7 1859.33   866.5 1856.53
   883.3 1858.48   908.7  1865.6     934 1866.22   955.1 1870.51     971 1875.55
#Mann= 11 ,-1,0
       0      .1       0      80     .07       0     170     .06       0
   271.2     .07       0     398    .045       0  463.05     .07       0
   471.2    .025       0  521.67     .03       0  591.67      .1       0
  703.81    .025       0  803.81      .1       0
Bank Sta=398,463.05
XS Rating Curve= 0 ,0
Exp/Cntr(USF)=0,0
Exp/Cntr=0.3,0.1

Type RM Length L Ch R = 1 ,1862    ,7.5,4.9,5.1
XS GIS Cut Line= 5
2191214.24826797649672.0045962482191455.34646715649664.843263599
 2191701.2188881649617.1010459392191844.44554108649521.616610619
2192135.67306881649619.488156822
#Sta/Elev= 30
       0 1872.36      66 1872.15      98 1870.97   241.2 1858.61   282.6  1858.3
   360.2 1859.81   368.4 1858.01   379.71851.065   384.9 1849.42   409.5 1849.25
   421.3  1849.3   425.4 1850.17  426.361851.117   433.6 1856.83     458  1859.2
   491.7 1857.92   594.7 1856.75   675.9 1857.03   709.9 1858.27   777.5 1858.72
     788 1858.19   802.8 1855.97   838.2 1856.88   849.2 1856.37   868.5 1861.42
     883 1864.02   904.1 1865.57   916.7 1870.09   950.1 1879.24     971 1886.38
#Mann= 10 ,-1,0
       0     .06       0      70      .1       0     220     .06       0
   261.2     .07       0   379.7    .045       0  426.36     .07       0
   461.2    .025       0  591.67      .1       0  693.81    .025       0
  793.81      .1       0
Bank Sta=379.7,426.36
XS Rating Curve= 0 ,0
Exp/Cntr(USF)=0,0
Exp/Cntr=0.3,0.1

Type RM Length L Ch R = 1 ,1857    ,48.4,43.9,43.3
XS GIS Cut Line= 6
2191179.61723296649687.4293190272191286.74418097649740.992793028
2191410.78591023649681.7910586062191813.92153035649597.217152288
2191892.85717625649559.1588944442192108.52063736649635.275410131
#Sta/Elev= 30
       0 1873.04    28.6 1872.44    31.5 1871.86    52.4 1863.64    72.2 1859.09
    94.1  1856.3   119.8 1854.65   227.7 1856.26   262.3 1857.66   424.4 1858.55
   434.6 1857.37   448.1 1850.78   454.8 1849.34   475.1 1849.25   483.4 1849.28
   487.5 1850.64   491.6 1855.63   495.7 1858.42   573.7 1857.42   798.9 1858.56
   822.9 1855.94   858.1 1855.95   887.5 1856.98   891.8 1857.93     902 1861.95
   917.2 1865.39   938.4 1867.52   951.2 1872.29   972.4    1877   985.5 1881.34
#Mann= 9 ,-1,0
       0     .06       0     110      .1       0  337.22     .07       0
   448.1    .045       0   487.5     .07       0  527.22    .025       0
  729.13      .1       0  739.13    .025       0  786.76      .1       0
#XS Ineff= 2 , 0
          320.13 1862.66  786.58         1860.96
Permanent Ineff=
       F       F
Bank Sta=448.1,487.5
XS Rating Curve= 0 ,0
Exp/Cntr(USF)=0,0
Exp/Cntr=0.3,0.1

Type RM Length L Ch R = 1 ,1813    ,226.1,255.1,260.3
XS GIS Cut Line= 6
2191141.55897512 649714.915838582191283.92505076649785.394093846
2191407.96678002649726.1923594232191811.10240014649641.618453105
2191890.03804604649603.5601952612192105.70150715649679.676710948
#Sta/Elev= 30
       0 1873.78    16.3 1872.67    30.5 1866.01    47.6 1859.88    84.2 1854.65
   114.1 1853.47   146.9 1855.54     321 1856.73   390.5 1858.42   418.1  1854.9
     460 1854.78   476.6 1850.45   496.1 1849.22   525.4 1849.47  532.381850.411
   549.9 1853.26   566.3 1854.11     603 1854.24   635.7 1858.03   672.3 1856.05
   795.3 1856.94   806.6 1856.05   891.4 1856.14   904.2 1860.25   925.4  1864.6
   944.9 1866.57   983.8 1877.69   997.5 1879.78    1006 1883.41  1024.5 1888.76
#Mann= 10 ,-1,0
       0      .1       0      50     .06       0     120     .07       0
  158.86      .1       0   466.3     .07       0   476.6    .045       0
  532.38     .07       0   566.3      .1       0   596.3    .025       0
  778.21      .1       0
#XS Ineff= 2 , 0
          228.38 1859.15  652.15         1862.34
Permanent Ineff=
       F       F
Bank Sta=476.6,532.38
XS Rating Curve= 0 ,0
Exp/Cntr(USF)=0,0
Exp/Cntr=0.3,0.1
